--- BACKCK2.prj (project) ---

Proj Title=BACKCK2
Current Plan=p01
Default Exp/Contr=0,0
English Units
Geom File=g01
Flow File=f01
Plan File=p01
BEGIN DESCRIPTION:
END DESCRIPTION:
DSS Export Rating Curves= 0
DSS Export Rating Curve Sorted= 0
DSS Export Volume Flow Curves= 0
DXF OffsetX= 0
DXF OffsetY= 0
DXF ScaleX= 0
DXF ScaleY= 0

--- BACKCK2.p01 (plan) ---

Plan Title=Floodplain
Program Version=4.00
Geom File=g01
Flow File=f01
K Sum by GR=0
Std Step Tol=0.01
Critical Tol=0.01
Num of Std Step Trials=20
Max Error Tol=0.3
Flow Tol Ratio=0.001
Split Flow NTrial=30
Split Flow Tol=0.02
Split Flow Ratio=0.02
Log Output Level=0
Friction Slope Method=1
Unsteady Friction Slope Method=2
Unsteady Bridges Friction Slope Method=1
Global Log Level=0
CheckData=False
Run HTab=0
Run UNet=0
Run PostProcess=0
UNET Theta=0
UNET Theta Warmup=0
UNET ZTol=0
UNET ZSATol=0
UNET MxIter=0
UNET MaxInSteps=0
UNET DtIC=0
UNET DtMin=0
UNET MaxCRTS=0
UNET WFStab=0
UNET SFStab=0
UNET WFX=0
UNET SFX=0
UNET DSS MLevel=0
UNET DZMax Abort=0
UNET Convert EG Bridges=0
UNET Use Existing IB Tables=0
UNET Froude Limit=0
UNET Froude Power=0
Write IC File=0
Echo Input=False
Echo Output=False
Write Detailed=0

--- BACKCK2.f01 (steady flow) ---

Flow Title=NFF Regression Equation
Program Version=4.10
Number of Profiles= 1
Profile Names=P100yr
River Rch & RM=BACKCK2,Main            ,28242.9
657.9741
River Rch & RM=BACKCK2,Main            ,26359.7
709.3858
River Rch & RM=BACKCK2,Main            ,25462.8
761.9025
River Rch & RM=BACKCK2,Main            ,22736.9
845.6347
River Rch & RM=BACKCK2,Main            ,19987.1
  939.31
River Rch & RM=BACKCK2,Main            ,14986.9
1037.066
River Rch & RM=BACKCK2,Main            ,11017.7
1150.948
River Rch & RM=BACKCK2,Main            ,10736.9
1283.518
River Rch & RM=BACKCK2,Main            ,9736.9
1302.281
River Rch & RM=BACKCK2,Main            ,7964.9
1441.296
River Rch & RM=BACKCK2,Main            ,438.3
1585.671
River Rch & RM=BACKCK2,Main            ,96.9
1589.426
Boundary for River Rch & Prof#=BACKCK2,Main            , 1
Up Type= 0
Dn Type= 3
Dn Slope=0.01026
DSS Import GetInterval= 0
DSS Import GetPeak= 0
DSS Import FillOption= 0

--- BACKCK2.g01 (geometry) ---

Geom Title=USGS 1m DEM
Program Version=4.10

River Reach=BACKCK2         ,Main
Reach XY= 30
     2164551.442      222581.189     2165166.025       222232.23
     2165794.497      222740.043      2166556.65        222879.8
     2167442.067      222615.043     2169554.914      222662.786
     2170002.831      222417.126     2171580.088      223207.925
     2172022.796      223785.182     2172008.907      225214.001
     2172442.067      225614.175     2172279.847      226550.048
     2173060.358      227845.696     2172571.237        228615.8
     2172981.006       229089.31     2173450.613      231181.079
     2174192.098       231486.78     2174143.967      232040.942
     2174781.384      232078.667     2175105.296      232601.609
     2175610.027      232766.817     2175754.421      233386.022
     2176367.122      233673.511     2176240.939      234258.894
      2176731.81      234362.094     2177175.821      234827.806
     2177598.998      234679.368      2178696.22      235527.458
      2179710.76      235239.568     2180229.083      235431.968

Type RM Length L Ch R = 1 ,28242.9 ,278.8,267.2,230.1
XS GIS Cut Line= 3
     2164549.777      222934.473      2164598.39      222707.032
     2164415.795      222175.909
#Sta/Elev= 30
       0 2284.57    42.6 2282.44    88.4 2282.02   163.8 2279.86   176.9 2278.55
   203.1 2278.58   252.2 2275.61   268.5 2271.29   294.6 2271.24   330.5 2268.99
   350.1  2269.5   357.4    2268   363.2  2266.3     373 2267.81   389.3 2268.99
   405.6 2268.19     422 2268.95   431.8 2267.78   444.8    2269   474.2 2268.13
   500.3 2271.07   542.8 2270.12   559.1 2273.84   585.2 2277.56     644 2297.84
   660.3 2305.79   699.5 2329.17   745.2 2353.49   771.4 2364.53   794.2 2371.88
#Mann= 3 ,-1 , 0
       0     .12       0   357.4    .045       0     373     .12       0
Bank Sta=357.4,373
XS Rating Curve= 0 ,0
Exp/Cntr=0.3,0.1

Type RM Length L Ch R = 1 ,27975.7 ,231.2,260.2,280.6
XS GIS Cut Line= 4
     2164925.333      222783.374     2164759.372      222479.666
     2164653.157      222408.303     2164459.548      222146.894
#Sta/Elev= 30
       0    2274    35.9 2271.74    71.8 2272.32   114.3  2272.1   189.4 2269.46
   293.8 2267.98   306.9 2266.57   342.8 2266.46   378.1 2265.48   397.3 2265.74
   403.7 2265.14   410.1  2263.3   422.9 2262.67   428.5 2263.34   432.5 2264.15
   445.3 2264.96   451.7 2266.58   503.3 2268.61   516.4 2272.89   526.1 2274.41
   561.9 2275.58   574.9 2277.28   581.4 2279.05   604.2 2288.45   646.5 2308.24
     679 2325.34   727.8 2353.38   760.3 2369.61   783.1 2379.83   799.4 2385.26
#Mann= 3 ,-1 , 0
       0     .12       0   410.1    .045       0   428.5     .12       0
Bank Sta=410.1,428.5
XS Rating Curve= 0 ,0
Exp/Cntr=0.3,0.1

Type RM Length L Ch R = 1 ,27715.5 ,438.2,457.7,450.4
XS GIS Cut Line= 3
     2164986.739      222748.522     2164880.524      222262.257
     2164953.546      221963.528
#Sta/Elev= 30
       0 2274.21    16.4 2272.07    65.5 2269.96    81.9 2268.36   101.5 2268.11
   137.5 2269.14   153.9 2267.95     262 2266.54   288.2  2265.6   307.8  2263.9
   360.2 2263.82   370.8  2261.2   376.6  2259.5   389.7 2260.98   409.3 2261.83
   422.4 2261.54   432.2 2262.46   445.3 2261.89   484.6 2262.25   487.9 2263.89
   497.7 2273.58   507.5 2281.56     537 2295.99   579.5 2310.28   615.5 2324.18
     645 2332.85   680.9 2347.85   716.9 2361.51     766 2382.49   805.3 2396.45
#Mann= 3 ,-1 , 0
       0     .12       0   370.8    .045       0   389.7     .12       0
Bank Sta=370.8,389.7
XS Rating Curve= 0 ,0
Exp/Cntr=0.3,0.1

Type RM Length L Ch R = 1 ,27257.7 ,259.4,270.8,282.9
XS GIS Cut Line= 2
     2165160.997      222690.436     2165273.851      221936.974
#Sta/Elev= 30
       0 2271.33    65.4  2263.4   127.5 2263.35   186.4 2262.14   199.5 2261.41
   212.5 2257.11   215.8  2256.8   251.8 2257.05   277.9 2256.23   297.6 2257.77
   349.9 2257.91   408.7 2259.61   425.1 2259.55   428.4 2259.09   444.7 2254.42
     448 2253.51   454.5 2253.19   461.3 2254.41   467.6 2257.92   477.4 2268.55
   483.9 2273.05   510.1  2285.8   536.2 2297.04   546.1 2301.86   575.5 2318.06
   595.1 2329.54   637.6 2351.92   676.8 2373.86   719.4 2392.58   761.9 2412.97
#Mann= 3 ,-1 , 0
       0     .12       0   444.7    .045       0   461.3     .12       0
Bank Sta=444.7,461.3
XS Rating Curve= 0 ,0
Exp/Cntr=0.3,0.1

Type RM Length L Ch R = 1 ,26986.9 ,262.3,280.4,329.9
XS GIS Cut Line= 3
       2165300.3      222705.864     2165482.458      222330.589
     2165644.307      222015.072
#Sta/Elev= 30
       0 2269.13    65.2  2258.4    91.2 2257.21   156.4 2257.08   179.2 2252.84
   224.9  2253.3   237.9 2252.45   250.9 2252.86   267.2 2254.53   293.3 2253.66
   316.1  2254.8   342.2 2254.33     378 2255.73   404.1 2252.43   409.6 2250.96
   417.2 2250.02   426.9 2250.94   433.4 2254.18   449.7 2254.71   456.2 2255.79
   459.4  2257.1   482.2 2274.45     492  2280.4   537.5 2299.63   592.8 2320.85
   635.1 2332.75   687.2 2346.09   729.5 2358.57   758.7 2369.23   771.8 2372.34
#Mann= 3 ,-1 , 0
       0     .12       0   409.6    .045       0   426.9     .12       0
Bank Sta=409.6,426.9
XS Rating Curve= 0 ,0
Exp/Cntr=0.3,0.1

Type RM Length L Ch R = 1 ,26706.5 ,357.7,346.8,285.9
XS GIS Cut Line= 2
      2165363.47      222756.821     2165965.907      222290.471
#Sta/Elev= 30
       0 2274.35    13.1 2270.83      49 2266.22    68.7 2262.57   104.6 2257.36
   117.7 2256.25   199.4  2254.3   232.2 2251.59   258.3 2251.81   274.7 2249.46
   297.6 2251.12     340 2250.81   346.7 2249.52   349.9 2247.86   353.1 2247.34
   366.2 2248.33   379.3 2249.35   402.2 2248.06   421.8 2250.56   477.4 2251.96
     497 2255.36   506.8 2256.06   519.9 2254.23   529.7 2259.56     533 2260.49
   565.7 2264.24   595.1 2266.28   608.2 2268.09   647.4 2279.34   761.8 2301.38
#Mann= 3 ,-1 , 0
       0     .12       0   346.7    .045       0   366.2     .12       0
Bank Sta=346.7,366.2
XS Rating Curve= 0 ,0
Exp/Cntr=0.3,0.1

Type RM Length L Ch R = 1 ,26359.7 ,198,189.5,180.1
XS GIS Cut Line= 2
     2165683.774      222957.633     2165970.886      222298.769
#Sta/Elev= 30
       0 2315.85    19.6 2313.29    35.9 2309.58    91.5 2292.35   120.9 2281.61
   169.9 2261.42   186.2 2251.94   192.7 2249.32   212.3 2248.12   222.1  2245.6
  234.612245.056   235.2 2244.94   238.5 2243.67     245 2243.35   254.8 2244.49
   274.4 2246.36   290.8 2245.77   313.6 2247.59   346.3  2247.8  385.252246.657
   398.6 2248.18   411.6 2248.68   509.6 2248.48     526 2252.18   561.9 2256.29
   594.6 2263.57   627.2 2278.04   653.4 2286.85   682.8 2293.99   718.7 2301.08
#Mann= 5 ,-1 , 0
       0     .12       0  234.61     .08       0   235.2    .045       0
   254.8     .08       0  385.25     .12       0
Bank Sta=235.2,254.8
XS Rating Curve= 0 ,0
Exp/Cntr=0.3,0.1

Type RM Length L Ch R = 1 ,26170.2 ,210.1,208.6,200.1
XS GIS Cut Line= 2
     2165894.544      223120.275     2166030.632      222351.876
#Sta/Elev= 30
       0 2406.23      23 2401.53    49.2 2393.56      82 2380.25   121.3 2360.94
   252.5 2289.11   278.7 2271.92   295.1 2259.48   321.3  2244.2   331.2 2242.71
     341 2243.84   354.1 2243.28   367.2 2244.13   380.3 2242.71   390.2 2240.68
   396.7 2241.44   399.9 2243.65   406.6 2245.36  415.212245.574   468.9 2244.98
   491.8 2242.71   501.7 2245.89   557.4 2245.14     5862245.961     623 2245.63
   665.6 2246.79   685.3 2249.62   704.9 2257.35   744.3 2279.89   780.4 2296.81
#Mann= 5 ,-1 , 0
       0     .12       0   380.3    .045       0   399.9     .12       0
  415.21     .08       0     586     .12       0
#XS Ineff= 2 , 0
                          413.77          2245.6
Permanent Ineff=
       F       F
Bank Sta=380.3,399.9
XS Rating Curve= 0 ,0
Exp/Cntr=0.3,0.1

Type RM Length L Ch R = 1 ,25961.6 ,230,224.8,221.5
XS GIS Cut Line= 2
     2166070.462      223184.999     2166181.656       222419.92
#Sta/Elev= 30
       0 2460.08     9.8 2455.41    26.2 2445.73    52.4 2431.48   212.9 2336.08
   281.7 2297.35   298.1 2284.94   337.4 2250.68   347.2 2240.89   353.7 2238.72
   360.4 2238.13   373.4 2238.87   383.3 2240.67   393.1 2240.13   402.9 2241.71
   419.3 2241.38   435.7 2242.73   465.2 2242.02   478.3 2242.41   497.9 2241.93
   520.9 2242.58   543.8    2242   556.9 2243.04   566.7 2242.82   589.7 2243.89
   651.9 2243.19   678.1 2243.54   750.2 2247.03   763.3 2249.11   773.1  2252.3
#Mann= 3 ,-1 , 0
       0     .12       0   353.7    .045       0   373.4     .12       0
#XS Ineff= 2 , 0
                          406.78         2241.84
Permanent Ineff=
       F       F
Bank Sta=353.7,373.4
XS Rating Curve= 0 ,0
Exp/Cntr=0.3,0.1

Type RM Length L Ch R = 1 ,25736.9 ,285.1,274.1,259.6
XS GIS Cut Line= 3
     2166342.693      223213.718     2166342.693      222850.286
     2166367.397      222483.899
#Sta/Elev= 30
       0 2434.66     9.8 2434.92    19.6 2433.24      36 2427.63    52.4 2420.12
    85.1 2402.92   163.7 2359.07   307.8  2280.4   317.6 2273.94     334 2260.67
   347.1 2247.64   353.6 2238.82   355.9 2236.75   356.9 2235.85   360.2 2235.12
   373.3 2235.91   389.7 2238.16   409.72237.899   425.7 2237.63     452 2239.45
   461.8 2239.04   484.8 2240.35   501.1 2239.73  512.832240.434   527.4  2241.1
     547 2240.21   553.6 2241.05   665.1 2245.19   701.1 2247.36   730.6 2251.98
#Mann= 5 ,-1 , 0
       0     .12       0   355.9    .045       0   373.3     .12       0
   409.7     .08       0  512.83     .12       0
#XS Ineff= 2 , 0
                          450.95         2242.41
Permanent Ineff=
       F       F
Bank Sta=355.9,373.3
XS Rating Curve= 0 ,0
Exp/Cntr=0.3,0.1

Type RM Length L Ch R = 1 ,25462.8 ,201.3,203.7,205.3
XS GIS Cut Line= 3
     2166392.426      223196.617      2166629.75      222936.058
     2166492.415      222490.011
#Sta/Elev= 30
       0 2412.72    19.6 2406.78    55.5 2393.95    91.4 2379.32   143.6 2355.98
   303.5 2281.97   342.6  2265.6   368.8 2258.55   401.4 2247.16   411.2 2242.19
   424.9 2233.34   427.5 2232.06   430.8  2231.7   440.6 2231.88   443.8 2232.62
   450.4  2234.1   463.4 2234.96   476.5 2233.55   486.2 2236.05     496 2235.88
   502.6 2235.05   522.2 2234.99     545 2237.62   564.6 2236.87   574.4 2238.38
   600.5 2240.31   626.6 2241.13   665.8 2243.49     731 2245.59   819.2 2249.93
#Mann= 3 ,-1 , 0
       0     .12       0   424.9    .045       0   443.8     .12       0
#XS Ineff= 2 , 0
                          486.56         2236.08
Permanent Ineff=
       F       F
Bank Sta=424.9,443.8
XS Rating Curve= 0 ,0
Exp/Cntr=0.3,0.1

Type RM Length L Ch R = 1 ,25259   ,298.6,304.5,310.2
XS GIS Cut Line= 3
     2166994.864      223128.573     2166784.094      222794.992
     2166691.156      222434.857
#Sta/Elev= 30
       0 2356.15     6.5 2354.03    19.6 2347.45    35.9 2346.41    39.1 2345.32
    55.4 2336.04   104.4 2314.58   182.6 2277.95   198.9 2270.95   221.8 2263.34
   234.8 2259.97   260.9 2255.68   316.3  2244.4   332.6 2242.94   352.2 2242.38
   381.5 2233.12   407.6  2232.1   420.7 2230.02   430.5 2229.79   440.3 2228.76
   443.5 2228.82   448.3 2230.59   453.3 2232.62   469.6 2232.07     499 2232.89
   525.1 2234.67   639.3 2237.44   675.2 2243.43   740.4 2249.04   766.5 2253.68
#Mann= 3 ,-1 , 0
       0     .12       0   430.5    .045       0   448.3     .12       0
#XS Ineff= 2 , 0
                          453.86         2234.38
Permanent Ineff=
       F       F
Bank Sta=430.5,448.3
XS Rating Curve= 0 ,0
Exp/Cntr=0.3,0.1

Type RM Length L Ch R = 1 ,24954.5 ,227.9,225.8,221.8
XS GIS Cut Line= 3
     2167136.356      223107.489     2167056.061      222792.819
      2167032.19      222345.771
#Sta/Elev= 30
       0 2379.18    39.4 2362.82    95.1 2337.49   101.7 2333.67   108.2 2328.32
   111.5    2327   121.4 2325.89   124.6 2324.41   134.5 2317.78   147.6 2310.56
   203.4 2281.98     269 2255.49   321.5 2238.76   341.1 2230.01   349.8 2227.36
   360.7 2225.65   367.2 2227.18   383.6 2228.57   429.3 2228.16  446.642229.286
   501.2 2229.02   530.6 2229.91  593.972227.098   625.4  2224.8     645 2225.37
   658.1 2228.68   674.4 2228.94   703.8 2231.54   723.4  2234.8   772.4 2240.75
#Mann= 5 ,-1 , 0
       0     .12       0   349.8    .045       0   367.2     .12       0
  446.64     .08       0  593.97     .12       0
#XS Ineff= 2 , 0
                          452.28          2229.6
Permanent Ineff=
       F       F
Bank Sta=349.8,367.2
XS Rating Curve= 0 ,0
Exp/Cntr=0.3,0.1

Type RM Length L Ch R = 1 ,24728.7 ,231.4,241.8,249.8
XS GIS Cut Line= 2
     2167335.083      223087.082      2167199.29      222311.048
#Sta/Elev= 30
       0  2399.1     9.8 2394.76    98.1 2348.38   156.9 2314.32   163.4 2309.74
     170 2303.72   179.8 2301.86   183.1 2300.56   199.4 2288.19   251.7  2257.1
   268.1 2250.14   294.2    2241   313.8 2229.39   320.4 2226.51   333.4 2226.25
   355.7    2224   362.9 2224.17   372.7 2222.41   379.2 2224.31     389 2225.82
   405.4 2225.46   441.3 2227.14   526.3 2227.86  601.762227.283   630.9 2226.93
   666.9 2228.35   712.6 2232.85   735.5 2238.65   768.2 2239.38   787.8 2241.76
#Mann= 4 ,-1 , 0
       0     .12       0   355.7    .045       0   379.2     .08       0
  601.76     .12       0
Bank Sta=355.7,379.2
XS Rating Curve= 0 ,0
Exp/Cntr=0.3,0.1

Type RM Length L Ch R = 1 ,24486.9 ,287.6,290.4,289.7
XS GIS Cut Line= 3
     2167445.261      223059.613     2167468.283      222618.515
     2167484.169      222267.024
#Sta/Elev= 30
       0 2376.97    58.9 2346.61   147.2 2299.21   153.8 2295.33   163.6 2286.74
   166.9 2284.97   176.7 2283.22     180 2281.57     193 2268.92   225.8  2240.2
   248.7 2223.24   255.2    2222   343.5 2224.69   350.1 2224.34   360.42221.838
   418.8 2223.25   428.6 2223.04   434.2 2221.39   441.7 2220.01   451.5 2221.58
   461.2 2224.01  480.572224.362   594.8 2222.09   627.4 2223.22   650.2 2222.33
     686 2224.22   712.1 2228.57     761 2232.95     774 2236.43   793.6 2246.25
#Mann= 5 ,-1 , 0
       0     .12       0   360.4     .08       0   434.2    .045       0
   451.5     .08       0  480.57     .12       0
#XS Ineff= 2 , 0
          343.53  2224.7  487.74         2224.53
Permanent Ineff=
       F       F
Bank Sta=434.2,451.5
XS Rating Curve= 0 ,0
Exp/Cntr=0.3,0.1

Type RM Length L Ch R = 1 ,24196.5 ,237.6,233.3,229.9
XS GIS Cut Line= 2
     2167648.749      223088.742     2167703.516      222297.109
#Sta/Elev= 30
       0 2337.66    52.5 2330.18    75.4 2324.98   104.9 2315.78   193.5 2281.94
   219.7 2270.89   236.1    2263   298.4 2227.43   308.2 2223.43   321.3 2221.96
   326.2 2219.43   331.2 2217.11   337.7 2216.68   350.9 2219.17   377.1 2220.46
  435.562220.198   501.7 2219.13   527.9 2220.57   544.3 2219.06   567.3 2221.16
   574.42220.691   596.8  2220.7   606.6 2219.17   616.5 2220.44   659.1 2220.45
   665.6 2222.73   675.5  2228.3   691.9 2233.17   777.1 2239.13   793.5 2242.55
#Mann= 5 ,-1 , 0
       0     .12       0   326.2    .045       0   350.9     .12       0
  435.56     .08       0   574.4     .12       0
#XS Ineff= 2 , 0
                          568.65         2221.18
Permanent Ineff=
       F       F
Bank Sta=326.2,350.9
XS Rating Curve= 0 ,0
Exp/Cntr=0.3,0.1

Type RM Length L Ch R = 1 ,23963.2 ,323.4,318.4,311.4
XS GIS Cut Line= 3
     2167919.805      223093.951     2167902.308      222730.372
     2167899.167      222366.221
#Sta/Elev= 30
       0 2413.84    45.9 2390.76    85.3 2369.55   147.6 2333.93   203.3 2300.74
   219.7 2289.57   275.5 2244.02   298.4 2229.11   311.5 2222.66   321.4 2220.43
   331.2 2215.96   344.3 2214.66   354.2 2213.64     364 2214.48   396.8 2218.02
   413.2 2216.86   432.9    2218   455.9 2216.07   472.3 2216.92  482.852215.659
   495.2 2215.31  520.932217.142   537.9 2215.37   554.3 2217.43  595.592218.369
   636.3 2219.55   642.9    2221   659.3 2226.69  702.752229.521   728.2  2233.1
#Mann= 7 ,-1 , 0
       0     .12       0   344.3    .045       0     364     .12       0
  482.85     .08       0  520.93     .12       0  595.59     .08       0
  702.75     .12       0
Bank Sta=344.3,364
XS Rating Curve= 0 ,0
Exp/Cntr=0.3,0.1

Type RM Length L Ch R = 1 ,23644.8 ,194.3,195.3,193.9
XS GIS Cut Line= 2
     2168287.698      223065.508     2168148.291      222355.195
#Sta/Elev= 30
       0 2445.75   104.8 2381.48   127.7  2366.1   160.5 2345.76   180.2 2331.41
   199.8 2318.84   232.6 2296.45   343.9 2214.62   347.2 2212.36     357  2208.9
   360.3 2208.42   374.7 2208.79   383.2 2210.46   389.8 2213.81     393 2214.56
     416  2212.6  469.182211.087   501.1 2210.47     511 2211.31   520.8 2210.46
   540.4  2212.8   579.8 2212.56   586.3 2213.55   609.2 2214.05   658.4 2218.98
   668.2  2219.4   694.4 2227.53   704.2 2231.84     714 2234.77   723.9 2239.23
#Mann= 4 ,-1 , 0
       0     .12       0     357    .045       0   374.7     .12       0
  469.18     .07       0
Bank Sta=357,374.7
XS Rating Curve= 0 ,0
Exp/Cntr=0.3,0.1

Type RM Length L Ch R = 1 ,23449.5 ,208,212.6,220.4
XS GIS Cut Line= 3
     2168468.857      223023.551     2168407.222      222664.948
     2168324.449      222309.673
#Sta/Elev= 30
       0 2423.31    19.7 2411.07    52.4  2388.3      82 2369.55    91.8  2362.4
   150.8 2325.06   213.1 2284.03   281.9 2240.67     318 2216.32   324.5 2210.37
   327.8 2208.64   347.5 2208.76   354.8 2207.25   357.3  2206.3   363.9 2205.72
   373.6 2207.03   383.4 2206.78     403 2209.71  408.81 2209.75   477.9 2210.04
   494.1 2211.14   539.7 2211.46   552.8 2213.77   565.8 2213.72   598.4 2218.46
   637.4 2225.88     657 2231.96  677.092240.082   696.1 2247.05   728.6 2260.55
#Mann= 5 ,-1 , 0
       0     .12       0   354.8    .045       0   373.6     .12       0
  408.81     .07       0  677.09     .12       0
#XS Ineff= 2 , 0
                          407.33         2210.91
Permanent Ineff=
       F       F
Bank Sta=354.8,373.6
XS Rating Curve= 0 ,0
Exp/Cntr=0.3,0.1

Type RM Length L Ch R = 1 ,23236.9 ,254.1,249.3,239
XS GIS Cut Line= 3
     2168631.246      223011.898     2168605.636      222641.085
     2168605.636      222278.443
#Sta/Elev= 30
       0 2381.57      13 2374.51    29.3 2363.48    42.4 2356.13   127.2 2303.89
   208.7 2251.94   221.7 2242.87   234.8  2234.9   257.6 2218.24   270.6 2207.13
   273.9 2206.19   290.2  2206.6   303.2 2204.16   316.3 2206.37   345.6 2206.45
   364.2 2204.88     375 2203.94   381.5 2204.78   401.1 2205.95  419.972209.578
   515.4 2216.35   538.3 2216.49   551.4 2217.65   567.7 2216.58     5912224.652
   610.2 2233.64   633.1 2246.74   688.6 2272.26   714.7 2285.69   734.3 2294.71
#Mann= 5 ,-1 , 0
       0     .12       0   364.2    .045       0   381.5     .12       0
  419.97     .07       0     591     .12       0
Bank Sta=364.2,381.5
XS Rating Curve= 0 ,0
Exp/Cntr=0.3,0.1

Type RM Length L Ch R = 1 ,22987.6 ,245.2,250.7,256.3
XS GIS Cut Line= 3
     2168920.009      222944.356     2168833.709      222564.306
     2168850.305      222225.746
#Sta/Elev= 30
       0 2340.63    39.3 2313.52    55.7 2303.11    78.6 2286.89   127.7 2255.22
     167 2232.24   219.4 2204.66   222.7 2203.46   229.2 2202.92   239.1 2203.66
   248.9    2203   271.8 2203.07   288.2  2204.1   314.4 2204.41   317.7 2204.24
   327.5 2201.93   335.9 2201.78   347.2 2200.29     357  2200.7   360.2 2201.75
   383.2 2207.64   415.8 2211.42  443.062218.493   461.4 2222.27   516.8 2230.43
   533.1 2230.41   542.9 2232.92  551.382233.536   640.7 2242.35   728.7 2249.86
#Mann= 5 ,-1 , 0
       0     .12       0   335.9    .045       0   360.2     .12       0
  443.06     .07       0  551.38     .12       0
Bank Sta=335.9,360.2
XS Rating Curve= 0 ,0
Exp/Cntr=0.3,0.1

Type RM Length L Ch R = 1 ,22736.9 ,233.4,250,270
XS GIS Cut Line= 3
       2169095.8      222907.173     2169051.607      222533.595
      2169020.17      222164.196
#Sta/Elev= 30
       0 2312.43    29.4 2292.01    55.6 2275.23    78.5 2261.98   130.8 2235.65
   153.7 2225.27   196.3 2207.58   212.6 2204.46   232.2 2202.58   281.3 2201.98
     350 2202.39   359.8 2199.43   366.4 2194.72   369.6 2193.48   376.2 2193.19
   385.9  2194.1   389.2 2195.99     399 2205.59   408.7 2210.51   434.7 2214.32
   473.7 2225.85   486.8 2228.26     503 2229.77     529 2230.21   571.3 2233.62
   581.1 2235.01   603.8 2235.35   613.6 2236.74   688.4 2242.54   746.9 2248.51
#Mann= 3 ,-1 , 0
       0     .12       0   366.4    .045       0   385.9     .12       0
Bank Sta=366.4,385.9
XS Rating Curve= 0 ,0
Exp/Cntr=0.3,0.1

Type RM Length L Ch R = 1 ,22486.9 ,277,263.6,244.3
XS GIS Cut Line= 3
     2169164.553      222916.287       2169282.1       222563.69
     2169438.776      222233.613
#Sta/Elev= 30
       0 2321.51      13 2311.73    58.7  2279.6   110.8 2244.08   146.7 2220.88
   172.8 2206.48   179.3 2203.73   189.1 2201.04   198.9 2200.31   247.8    2200
   303.2 2198.32   342.3 2199.11   364.2 2192.51   374.9 2190.75   381.5 2191.22
   384.7 2192.26   394.5 2198.84   404.3 2201.34   417.4 2201.59   440.2 2203.65
   498.9 2210.36   534.8 2212.22   590.2 2212.06   619.6 2208.62   629.4 2206.83
   632.7 2206.93   645.7 2210.41   668.5 2213.86   697.9 2215.18     737 2219.46
#Mann= 3 ,-1 , 0
       0     .12       0   364.2    .045       0   384.7     .12       0
Bank Sta=364.2,384.7
XS Rating Curve= 0 ,0
Exp/Cntr=0.3,0.1

Type RM Length L Ch R = 1 ,22223.3 ,256.1,241,226.1
XS GIS Cut Line= 2
     2169537.383      222975.889     2169508.044      222254.186
#Sta/Elev= 30
       0 2394.17    19.6 2384.57    58.8 2361.85    81.7  2346.7   117.7 2325.06
   130.7 2315.29   166.7 2292.57   192.8 2274.69   215.7 2257.54   254.9 2226.55
   294.2 2193.77   297.4  2191.8     305 2189.38   313.8 2188.05   320.3 2188.28
   326.8 2189.82   336.6  2194.1   369.3 2192.93   421.6 2205.91  435.142206.943
   441.2 2206.59     451 2203.95   457.6 2203.22     536 2204.93  562.082204.263
   575.2 2204.06   594.8 2207.22   627.5 2208.63   663.5 2211.56   722.3 2217.64
#Mann= 5 ,-1 , 0
       0     .12       0     305    .045       0   326.8     .12       0
  435.14     .04       0  562.08     .12       0
Bank Sta=305,326.8
XS Rating Curve= 0 ,0
Exp/Cntr=0.3,0.1

Type RM Length L Ch R = 1 ,21982.3 ,240.5,242.4,243.7
XS GIS Cut Line= 3
     2169691.726      222916.143     2169758.111      222607.456
     2169574.931      222234.637
#Sta/Elev= 30
       0 2339.81    71.6 2293.76   117.2 2260.79   146.5 2238.35     179 2215.44
   188.8 2209.02   211.6 2196.29   218.1 2194.18   224.6 2193.24   286.4 2192.29
     306 2190.11   322.3 2190.22   338.6 2187.08   351.7 2186.46   357.2 2185.21
   361.5 2184.21   368.1 2183.82   374.6 2185.35   381.2 2189.51   384.4 2190.76
   410.6 2192.69     4312193.251  450.322194.454   541.4 2197.27   580.7  2200.1
   603.6 2203.54     633  2210.1   662.4 2214.39   708.2 2220.27   731.1 2221.78
#Mann= 5 ,-1 , 0
       0     .12       0   357.2    .045       0   374.6     .12       0
     431     .06       0  450.32     .12       0
Bank Sta=357.2,374.6
XS Rating Curve= 0 ,0
Exp/Cntr=0.3,0.1

Type RM Length L Ch R = 1 ,21739.9 ,227.5,264.3,293.6
XS GIS Cut Line= 3
     2169811.218      222904.526     2169958.923      222479.666
     2169798.846      222117.882
#Sta/Elev= 30
       0 2304.46    29.3 2283.64      75 2247.92   114.1 2219.12   143.4 2199.73
   153.2 2194.57     163 2191.35     176 2189.71   195.6  2190.9   218.4 2189.74
   231.4  2190.6   466.2 2185.96   485.8 2182.68   502.1 2180.98   508.6 2182.49
   521.7 2196.07   528.3 2198.21   541.4 2197.31     561 2190.85   567.5 2190.64
   619.8 2196.18   636.2 2200.64   655.8 2199.94   737.5  2205.3   744.1 2206.59
   760.4 2213.37   786.6 2216.54   809.4 2217.93   835.6 2216.78   845.4 2218.69
#Mann= 3 ,-1 , 0
       0     .12       0   485.8    .045       0   508.6     .12       0
Bank Sta=485.8,508.6
XS Rating Curve= 0 ,0
Exp/Cntr=0.3,0.1

Type RM Length L Ch R = 1 ,21475.6 ,253,256.5,257.3
XS GIS Cut Line= 2
     2169955.082      222917.393     2170251.014      222195.873
#Sta/Elev= 30
       0 2273.96    81.9 2209.62    91.8 2203.06   114.7 2190.49   134.3 2186.76
     272 2187.26   294.9 2185.86   321.1 2186.58   330.9 2185.25   344.2 2178.88
   350.6 2177.71   363.7 2178.56   383.4 2182.47   399.8 2181.41   416.1 2184.18
   432.5 2184.54   455.5 2189.91   465.3 2191.03   553.8 2192.39   583.2 2194.76
   599.6 2197.74     616 2198.61   625.8 2201.26   642.2 2203.15   668.4 2208.18
   681.6 2211.81   694.7 2217.29   707.8 2217.61   717.6 2222.07   779.8 2237.41
#Mann= 3 ,-1 , 0
       0     .12       0   344.2    .045       0   363.7     .12       0
Bank Sta=344.2,363.7
XS Rating Curve= 0 ,0
Exp/Cntr=0.3,0.1

Type RM Length L Ch R = 1 ,21219.1 ,236.1,232.2,226.8
XS GIS Cut Line= 3
     2170134.841      222975.889     2170324.037       222590.86
     2170543.165      222346.871
#Sta/Elev= 30
       0 2257.26      36 2231.27    55.7 2215.82    75.3  2202.7      95 2191.04
   108.1 2186.71   124.4  2184.8   199.8 2183.42   222.7 2184.19   235.8 2182.79
   284.9 2185.12   320.9 2183.83   353.7 2184.29   360.2 2183.42   383.2 2176.12
     393 2174.86   406.1 2176.44   415.9 2180.97   425.7  2182.6   445.4  2191.5
   458.5  2193.6   494.6 2196.24   540.5 2197.02   553.6 2194.96   566.7 2195.56
   586.4 2193.09   625.8 2196.27   642.2 2200.58     675 2211.51     757 2245.75
#Mann= 3 ,-1 , 0
       0     .12       0   383.2    .045       0   406.1     .12       0
Bank Sta=383.2,406.1
XS Rating Curve= 0 ,0
Exp/Cntr=0.3,0.1

Type RM Length L Ch R = 1 ,20986.9 ,250.6,250,248
XS GIS Cut Line= 3
     2170389.366      223076.593     2170509.372      222732.944
     2170629.377      222389.295
#Sta/Elev= 30
       0 2252.57    26.2 2234.06    65.6 2207.88   101.7 2187.41   121.3 2179.96
   127.9 2179.28     164 2179.22   249.2  2180.5   291.9 2180.15   314.8  2178.2
     341 2178.37   344.3 2177.74   350.9 2174.46   354.2 2172.93     364 2172.57
   371.5 2174.08   393.5  2177.8   406.6  2182.3   432.9 2181.92   449.3 2189.16
   459.1 2191.68   508.3 2194.92   521.4 2196.83   541.1 2196.26   550.9 2198.34
   593.6 2200.93     646 2206.42   655.9 2208.71     669 2213.09     728 2237.16
#Mann= 3 ,-1 , 0
       0     .12       0   350.9    .045       0   371.5     .12       0
Bank Sta=350.9,371.5
XS Rating Curve= 0 ,0
Exp/Cntr=0.3,0.1

Type RM Length L Ch R = 1 ,20736.9 ,258,249.6,242
XS GIS Cut Line= 3
     2170624.426      223178.361     2170750.685      222797.215
     2170852.591      222447.826
#Sta/Elev= 30
       0 2236.13    55.5 2192.96    75.1 2179.43    84.9 2176.16   114.2 2174.72
   130.6 2176.27   176.3 2176.86   205.6 2175.02   270.9 2176.42   336.2 2175.63
   355.8 2173.46   378.7 2172.87   388.5 2171.65   401.5 2169.84   411.4 2171.59
   421.2 2175.95   437.6 2179.43   470.4 2180.95   486.8 2177.29     513 2184.99
   526.1 2182.53   532.7 2182.57   552.3 2188.65     572 2188.42   598.2  2190.9
   627.8 2192.01   650.7 2195.13   696.6 2198.74   719.6 2203.88   765.5  2217.5
#Mann= 3 ,-1 , 0
       0     .12       0   388.5    .045       0   411.4     .12       0
Bank Sta=388.5,411.4
XS Rating Curve= 0 ,0
Exp/Cntr=0.3,0.1

Type RM Length L Ch R = 1 ,20487.3 ,191.6,216.8,241.5
XS GIS Cut Line= 3
     2170908.219      223246.405      2170986.22      222894.568
     2171022.472      222489.016
#Sta/Elev= 30
       0 2200.37    3.052198.327    22.9 2185.46    45.9 2171.55    52.4 2170.34
    59.8 2170.46   101.6 2169.58   163.8 2170.82   176.9  2170.1   268.6 2170.93
   278.5 2171.67   311.2  2172.1   330.9 2169.82   350.6 2170.98   366.9 2170.49
   386.4 2168.97   396.2 2166.94     406 2165.57   412.5 2167.13   415.8 2169.09
   425.5 2177.62   428.8 2179.14   441.8 2181.89   461.4 2183.43   559.1 2187.93
   578.6 2187.23     621 2193.14   708.9 2208.04     748 2213.07   767.6 2217.87
#Mann= 5 ,-1 , 0
       0     .12       0    3.05     .08       0    59.8     .12       0
   396.2    .045       0   412.5     .12       0
#XS Ineff= 2 , 0
          351.18 2171.02
Permanent Ineff=
       F       F
Bank Sta=396.2,412.5
XS Rating Curve= 0 ,0
Exp/Cntr=0.3,0.1

Type RM Length L Ch R = 1 ,20270.5 ,289,283.4,277.7
XS GIS Cut Line= 3
     2170976.263      223287.895     2171162.139      222952.654
     2171444.272      222650.606
#Sta/Elev= 30
       0 2209.52    39.3 2184.14    49.1 2176.66    55.7 2173.42    81.9 2170.72
  203.322169.102     249 2166.85   301.4 2167.28   337.4  2170.1   386.6 2169.51
   396.4 2168.52   416.1 2163.52   422.7 2162.68   435.8 2163.74   448.9  2169.8
   481.7  2172.2   501.4 2178.08     508 2178.82   521.1 2174.25   527.7 2174.24
   540.8 2178.11   553.9 2177.38   563.7 2182.36     567 2182.95   583.4 2183.19
   603.1 2188.29   645.8 2192.19   714.6 2203.21   744.2 2209.58   796.6 2227.98
#Mann= 4 ,-1 , 0
       0     .08       0  203.32     .12       0   416.1    .045       0
   435.8     .12       0
#XS Ineff= 2 , 0
          335.94 2170.36
Permanent Ineff=
       F       F
Bank Sta=416.1,435.8
XS Rating Curve= 0 ,0
Exp/Cntr=0.3,0.1

Type RM Length L Ch R = 1 ,19987.1 ,266.7,300.5,333.4
XS GIS Cut Line= 3
     2171197.844      223405.522     2171433.955      223061.772
     2171611.038      222787.466
#Sta/Elev= 30
       0 2207.58    32.6 2196.66    65.2 2182.54    81.4 2177.38    86.72176.574
    97.7 2175.27   149.9  2172.9     202 2171.37   211.8 2170.47   224.8 2170.86
  252.112169.208   322.6 2166.64   342.1 2164.12   361.6 2159.97   371.4  2158.8
   381.6 2160.22     404 2164.31   430.1 2164.42   482.3 2167.18   492.1 2169.56
   508.4 2175.05   544.4 2183.58   557.4 2184.36     577 2183.34   586.8 2187.36
   596.6 2188.77   661.9 2194.86     675 2198.66   710.9 2215.01   743.5 2226.17
#Mann= 5 ,-1 , 0
       0     .12       0    86.7     .08       0  252.11     .12       0
   361.6    .045       0   381.6     .12       0
Bank Sta=361.6,381.6
XS Rating Curve= 0 ,0
Exp/Cntr=0.3,0.1

Type RM Length L Ch R = 1 ,19686.6 ,482.7,449.7,394.7
XS GIS Cut Line= 4
     2171256.736      223462.154     2171490.741       223307.81
     2171641.765      223292.874     2171980.325      223110.317
#Sta/Elev= 30
       0 2221.26    61.9 2184.35   80.942174.431      88  2172.4     101 2170.72
   146.7 2168.15   159.7 2168.25   185.8 2165.45   228.2 2162.59   293.2 2161.46
   312.6 2160.08  359.372159.946   380.4 2158.41   393.3 2156.94     403 2157.36
   406.2 2158.31   412.7 2161.58   415.9 2162.13   490.8 2166.19   513.6  2170.3
   549.4 2173.16   572.2 2177.48   595.1 2176.92   601.6 2180.19   604.8 2180.68
   640.7 2182.75   712.4 2191.33     732  2196.1   784.1 2215.85   816.7 2225.43
#Mann= 5 ,-1 , 0
       0     .12       0   80.94     .08       0  359.37     .12       0
   380.4    .045       0   406.2     .12       0
Bank Sta=380.4,406.2
XS Rating Curve= 0 ,0
Exp/Cntr=0.3,0.1

Type RM Length L Ch R = 1 ,19236.9 ,234,250,265.3
XS GIS Cut Line= 3
     2171598.476      223817.943     2171833.178      223450.147
     2172035.874      223163.106
#Sta/Elev= 30
       0 2218.77    19.7 2204.76    62.3 2177.43    78.7 2168.66    88.6 2165.58
   150.9 2162.45   249.3  2160.3     269 2158.93   341.2 2158.66     374 2156.37
   387.1 2157.29   400.2 2157.16   423.2  2154.7   428.8 2153.29   442.8 2150.81
   449.3 2151.12   452.6 2152.47   462.3 2161.42   465.6 2162.85   491.6 2164.37
   533.9  2164.9   543.7 2165.78   559.9 2169.75     573 2170.51   582.7 2174.54
   595.7 2178.71     638 2189.46   693.3  2205.9   777.9 2238.54   787.7 2241.77
#Mann= 3 ,-1 , 0
       0     .12       0   428.8    .045       0   452.6     .12       0
Bank Sta=428.8,452.6
XS Rating Curve= 0 ,0
Exp/Cntr=0.3,0.1

Type RM Length L Ch R = 1 ,18986.9 ,233.1,250,268.4
XS GIS Cut Line= 3
     2171637.745      223872.249     2171939.523      223668.114
     2172254.222      223476.448
#Sta/Elev= 30
       0 2227.01    32.5 2205.16    68.3 2182.19    94.3 2167.16   100.8 2164.38
   110.6 2161.94   126.9 2160.44   159.4 2160.22   191.9 2157.56   341.6 2156.28
   348.1 2155.42   356.8 2150.94   361.1 2148.63   364.3 2147.97   380.6 2150.54
   393.7 2152.74   406.7 2158.29   426.3 2162.15   452.4 2166.06   471.9 2169.82
   488.2 2169.92     498 2174.09   511.1 2176.16   553.5 2192.69   582.8 2200.41
   602.4 2202.85   631.7 2205.01   670.8 2213.27   700.2  2217.7   732.8 2224.35
#Mann= 3 ,-1 , 0
       0     .12       0   356.8    .045       0   380.6     .12       0
Bank Sta=356.8,380.6
XS Rating Curve= 0 ,0
Exp/Cntr=0.3,0.1

Type RM Length L Ch R = 1 ,18736.9 ,236,238.7,240.5
XS GIS Cut Line= 3
     2171669.255      223945.801     2172035.114      223889.291
     2172397.549        223870.8
#Sta/Elev= 30
       0 2247.39    49.1 2217.81    78.6 2200.96     131 2173.63   150.7 2164.67
   163.8 2160.25   170.4  2158.9     190 2157.62   229.3 2153.46   288.3  2154.1
   327.6 2152.89   350.5 2153.45   357.1  2151.6   362.7 2147.83   366.9 2146.07
   370.2  2145.9   376.7 2146.11   383.3  2147.6   399.6 2151.03     429 2155.33
   438.9 2157.97   451.9 2159.01     465 2163.74   504.2 2170.77   523.9 2177.77
     550  2190.8   579.4 2204.23   621.9 2219.52   661.2 2230.29   733.1 2243.32
#Mann= 3 ,-1 , 0
       0     .12       0   362.7    .045       0   383.3     .12       0
Bank Sta=362.7,383.3
XS Rating Curve= 0 ,0
Exp/Cntr=0.3,0.1

Type RM Length L Ch R = 1 ,18498.2 ,259.3,261.3,257.1
XS GIS Cut Line= 3
     2171693.213      224233.871     2171980.325      224125.997
     2172386.684      224124.302
#Sta/Elev= 30
       0 2334.38      62 2294.16    97.9 2272.97   107.7 2266.46   117.5 2261.64
   127.2 2255.18   234.9 2190.96   251.2 2180.66   283.9 2162.25     310  2151.4
   319.8 2146.06   332.1 2143.43   342.8 2142.27   352.6 2143.73   362.4 2147.64
     369 2148.48   388.6 2149.55   411.6 2148.86   447.6 2150.18   467.3 2150.07
   503.3 2154.81     523 2162.95   542.7 2173.18     559 2182.44   572.2 2187.88
     582 2193.33   604.9 2202.83   627.9 2211.13   680.3 2225.98   713.1 2236.85
#Mann= 3 ,-1 , 0
       0     .12       0   332.1    .045       0   352.6     .12       0
Bank Sta=332.1,352.6
XS Rating Curve= 0 ,0
Exp/Cntr=0.3,0.1

Type RM Length L Ch R = 1 ,18236.9 ,240.2,235.2,231.8
XS GIS Cut Line= 3
     2171686.037      224382.197     2172076.316      224371.025
       2172434.2      224339.433
#Sta/Elev= 30
       0 2356.34    22.8 2344.15    65.1 2323.33    94.4  2307.5   143.2 2277.11
     205 2242.09     218 2234.19   276.6  2193.6   315.6    2168   325.4 2163.43
   344.9 2152.55   357.9  2148.7   370.9 2142.57   380.7  2141.1   387.2 2140.45
   403.5 2141.12   413.3 2145.28   416.6 2145.69     446 2147.31   462.3 2146.54
   472.1 2147.95   501.5 2149.64   511.3 2154.42   540.7 2175.95   563.5 2190.38
   576.6 2197.08   596.2 2205.27   641.9 2217.02   726.8 2229.43   749.7 2233.74
#Mann= 3 ,-1 , 0
       0     .12       0   380.7    .045       0   403.5     .12       0
Bank Sta=380.7,403.5
XS Rating Curve= 0 ,0
Exp/Cntr=0.3,0.1

Type RM Length L Ch R = 1 ,18001.7 ,236.7,253.3,269.8
XS GIS Cut Line= 4
     2171699.851      224547.537     2171981.992      224600.752
     2172138.816      224573.924     2172430.483      224606.911
#Sta/Elev= 30
       0 2342.39    29.4 2326.07      62 2304.73    97.9 2278.34   153.4 2234.68
   172.9 2218.65   202.3 2196.22   238.2 2170.52   264.3 2153.93   277.3 2147.99
   293.6 2145.91   332.6 2146.14   374.8  2145.3     378 2144.35   384.5 2140.39
   387.8 2139.19   397.5 2137.84   410.5 2136.97   420.2 2138.29   433.2  2142.4
   449.5  2141.4   462.5 2142.83   472.3 2147.06   488.6 2156.99   547.3 2198.89
   622.3    2247   658.2 2269.14   697.3 2291.68   720.2 2303.88   739.7  2313.2
#Mann= 3 ,-1 , 0
       0     .12       0   397.5    .045       0   420.2     .12       0
Bank Sta=397.5,420.2
XS Rating Curve= 0 ,0
Exp/Cntr=0.3,0.1

Type RM Length L Ch R = 1 ,17748.4 ,277.2,261.5,242.1
XS GIS Cut Line= 2
     2171681.596      224720.136      2172383.61       224914.31
#Sta/Elev= 30
       0 2303.14    39.2 2276.82      98 2239.76   127.4 2220.29   140.4 2210.53
     160 2199.22   179.6 2185.68   218.8  2161.4   228.6 2157.57   248.2 2152.99
   326.6 2146.13   333.2  2143.5   339.7 2137.41   346.2 2133.35   352.8 2132.69
   369.1  2133.5   378.9  2136.2   395.2 2138.58   421.4  2138.2   440.9 2141.25
     454 2141.04   463.8 2142.29   535.7  2140.7   574.9 2161.31   617.3 2186.71
   653.2 2204.84   676.1 2214.29   689.2 2218.24     699 2222.84   728.4 2233.57
#Mann= 3 ,-1 , 0
       0     .12       0   346.2    .045       0   369.1     .12       0
Bank Sta=346.2,369.1
XS Rating Curve= 0 ,0
Exp/Cntr=0.3,0.1

Type RM Length L Ch R = 1 ,17486.9 ,273.9,252.3,236.8
XS GIS Cut Line= 3
     2171627.373      225120.367     2171977.487      225066.124
     2172384.923      224968.299
#Sta/Elev= 30
       0 2220.96    29.5 2222.53    62.3 2218.98    75.4 2219.17   101.7  2217.3
   141.1 2215.98   150.9 2214.87     164 2211.71   193.6 2202.16   236.2 2183.75
   262.4 2174.02   288.7 2168.41   301.8  2164.1   321.5 2150.53   334.6 2137.53
   344.4  2130.2     351 2129.09   364.1 2129.74   409.9 2138.09   439.4 2139.54
   511.4 2139.11   537.6 2139.75   563.8 2141.65   635.8 2139.54   658.7 2140.43
   668.6 2145.23   678.4 2151.61   720.9 2183.95   756.9  2208.6   773.3 2218.44
#Mann= 3 ,-1 , 0
       0     .12       0   344.4    .045       0   364.1     .12       0
Bank Sta=344.4,364.1
XS Rating Curve= 0 ,0
Exp/Cntr=0.3,0.1

Type RM Length L Ch R = 1 ,17234.6 ,211.6,220.6,228.7
XS GIS Cut Line= 3
     2171850.137      225548.076     2172063.306      225294.361
      2172413.83      225028.715
#Sta/Elev= 30
       0 2356.02      39 2337.04    97.5 2306.29   198.2 2246.13   224.2 2228.34
   292.4 2178.55   305.4 2168.26   318.4 2155.78   337.9 2139.87   347.8 2128.45
   350.9 2126.17   357.4 2125.38   370.5 2126.98   383.5 2131.29     390 2132.31
   429.1 2132.86   530.1 2140.26     566 2144.21   582.2 2143.82   588.8 2145.62
   601.8 2145.96   618.1 2147.72   666.9  2148.6   676.7 2153.28   686.5 2160.66
   699.5 2166.19   709.3 2174.47   735.4 2193.04   754.9 2206.24   771.2 2215.87
#Mann= 3 ,-1 , 0
       0     .12       0   347.8    .045       0   370.5     .12       0
Bank Sta=347.8,370.5
XS Rating Curve= 0 ,0
Exp/Cntr=0.3,0.1

Type RM Length L Ch R = 1 ,17014   ,295,280.6,261.4
XS GIS Cut Line= 3
     2171931.881      225627.469     2172229.266      225403.895
     2172586.169      225245.874
#Sta/Elev= 30
       0 2356.04    26.1 2338.92    35.9 2333.49    71.8 2307.54   150.1 2253.17
   208.9 2209.65   264.4 2165.69   280.7 2151.95   300.2 2136.98   306.8  2133.9
   319.8  2131.9   329.6  2131.1   349.2  2131.3   378.6 2128.02   388.4 2125.66
   401.6  2123.5   404.8 2123.94   408.1 2125.55   424.5 2136.22     454 2138.57
   516.4 2146.16   526.2 2148.53   532.8 2151.06   542.6  2152.4   575.4 2162.64
   631.2 2174.02     641 2177.88     664  2189.3   719.7 2220.43   762.4 2238.27
#Mann= 3 ,-1 , 0
       0     .12       0   388.4    .045       0   408.1     .12       0
Bank Sta=388.4,408.1
XS Rating Curve= 0 ,0
Exp/Cntr=0.3,0.1

Type RM Length L Ch R = 1 ,16733.4 ,226.1,255.1,284.1
XS GIS Cut Line= 3
     2172026.107      225770.636     2172391.908      225614.665
     2172627.488      225302.895
#Sta/Elev= 30
       0 2337.93   123.9 2249.65   153.2 2227.53   185.8  2199.4   211.9  2178.4
   254.2 2146.23   273.8 2134.08   290.1 2129.23   309.7 2129.47   329.2 2126.97
   355.3 2127.38   368.3  2125.9   394.4 2125.94   426.6 2121.23   433.5 2120.04
   449.8 2121.59     453    2124   469.3 2144.26   485.6 2155.98   495.4 2159.22
   511.6 2158.97   518.2 2162.36   521.4 2162.73   550.7  2163.1   570.2 2165.65
   625.6 2185.22   671.2 2193.83   687.5 2200.58   742.8 2230.88   788.4 2250.22
#Mann= 3 ,-1 , 0
       0     .12       0   426.6    .045       0   449.8     .12       0
Bank Sta=426.6,449.8
XS Rating Curve= 0 ,0
Exp/Cntr=0.3,0.1

Type RM Length L Ch R = 1 ,16478.3 ,214.9,224,232
XS GIS Cut Line= 2
     2172039.221      225866.748     2172757.022      225749.093
#Sta/Elev= 30
       0 2348.76    26.2 2330.44    62.2 2303.89    91.7 2284.05   134.3 2253.08
   173.6  2221.9   288.3  2135.5   304.7 2126.03   311.3 2123.64     344 2124.49
   347.3 2123.33   353.9 2119.03   357.1 2117.47     367 2116.58   370.2 2116.65
   376.8  2119.2   399.7 2125.75     439  2133.6   458.7 2144.37   475.1  2145.9
   484.9 2152.75   494.8 2156.16   537.3 2164.54   566.8 2171.54   583.2 2176.38
   609.4 2187.37     652 2206.95   681.5 2217.36     711 2226.41   727.4 2229.78
#Mann= 3 ,-1 , 0
       0     .12       0   353.9    .045       0   376.8     .12       0
Bank Sta=353.9,376.8
XS Rating Curve= 0 ,0
Exp/Cntr=0.3,0.1

Type RM Length L Ch R = 1 ,16254.3 ,256.2,267.4,275
XS GIS Cut Line= 2
     2172036.523      226006.443     2172765.693      226054.805
#Sta/Elev= 30
       0 2354.64   30.192333.719  151.052247.728   252.3 2173.46   294.9 2139.93
   314.6 2125.61   321.2  2122.1   324.4 2121.38   340.8 2120.99   357.2  2116.6
     367 2114.65   376.9 2116.27     390 2118.95     426 2123.13   452.2 2124.92
   468.6 2127.69   478.4 2126.88     485  2127.1   511.2 2130.75   547.3 2133.87
   563.6 2136.65   573.5 2139.45   583.3  2143.4   593.1 2149.11     603 2150.82
   606.2 2152.56   612.8 2157.84     662 2189.15   704.6  2218.7   730.8 2235.67
#Mann= 5 ,-1 , 0
       0     .12       0   30.19     .08       0  151.05     .12       0
   357.2    .045       0   376.9     .12       0
Bank Sta=357.2,376.9
XS Rating Curve= 0 ,0
Exp/Cntr=0.3,0.1

Type RM Length L Ch R = 1 ,15986.9 ,266.4,250,236.9
XS GIS Cut Line= 3
     2172017.083      226159.687     2172362.425      226280.929
     2172717.574      226372.932
#Sta/Elev= 30
       0 2340.24    55.6 2301.25   120.9 2253.61   189.5 2199.01     219 2174.18
   248.4 2147.44   271.2 2129.92   277.8 2126.72   284.3 2125.11   297.4 2122.64
   313.7 2121.05   333.3 2115.45   343.1 2114.71   358.5 2110.81   372.6  2110.1
   382.4 2110.56   385.7 2110.87   398.8 2116.15   418.4 2118.23   438.1 2117.61
   513.4 2119.67   549.4 2135.31   562.5 2144.17   565.8 2145.42   575.6 2144.81
   578.9 2146.54     592 2157.22   657.5 2189.93   700.1 2208.51   732.9 2219.51
#Mann= 3 ,-1 , 0
       0     .12       0   358.5    .045       0   382.4     .12       0
Bank Sta=358.5,382.4
XS Rating Curve= 0 ,0
Exp/Cntr=0.3,0.1

Type RM Length L Ch R = 1 ,15736.9 ,269.5,250,234.6
XS GIS Cut Line= 3
     2171919.685      226539.325     2172271.355      226504.158
     2172693.847      226469.282
#Sta/Elev= 30
       0 2326.86    19.6 2311.43      72 2272.86     108 2248.23   150.5 2220.54
   163.6  2213.2   189.8 2200.41   248.7 2167.58   261.8 2162.18   271.6 2156.35
   294.5  2145.2   307.6 2136.76     324 2123.69   337.1 2109.16   340.3 2107.16
   353.4 2106.08   360.9 2106.78   389.3 2114.63   421.9 2115.24     435  2116.4
   454.5  2115.9     461 2117.53   490.4 2121.13   532.8 2123.49   581.7 2137.04
     611 2146.86   620.8 2148.32   679.5 2161.15   725.2 2163.04   777.4  2166.8
#Mann= 3 ,-1 , 0
       0     .12       0   340.3    .045       0   360.9     .12       0
Bank Sta=340.3,360.9
XS Rating Curve= 0 ,0
Exp/Cntr=0.3,0.1

Type RM Length L Ch R = 1 ,15486.9 ,232.6,250,256.2
XS GIS Cut Line= 3
     2172098.799      226930.487     2172397.968      226710.576
     2172720.986      226532.246
#Sta/Elev= 30
       0 2201.37    32.6 2178.21    78.2 2141.99   104.2 2123.68     114 2115.24
   117.2 2113.56     127 2111.12     140 2105.69   149.8 2105.22   185.6 2106.46
   218.2 2109.29   273.6 2110.94   299.6 2109.92   309.4 2108.21   325.7 2107.33
   335.5 2104.04   363.8 2100.31   377.8 2099.09   381.1 2099.32   384.4 2100.76
     404 2113.79   446.4 2144.57   462.7 2154.35     479 2162.61   495.4 2169.69
   531.3  2181.9   550.9 2186.14   590.1 2191.92   642.3 2197.43   740.3 2204.83
#Mann= 3 ,-1 , 0
       0     .12       0   363.8    .045       0   384.4     .12       0
Bank Sta=363.8,384.4
XS Rating Curve= 0 ,0
Exp/Cntr=0.3,0.1

Type RM Length L Ch R = 1 ,15236.9 ,274.2,250,233.6
XS GIS Cut Line= 3
     2172128.161       226997.24     2172503.593      226932.273
     2172849.765      226821.789
#Sta/Elev= 30
       0 2194.77    32.6 2171.12    48.8 2156.56   104.2 2109.79   110.7 2106.33
   123.8 2103.43   133.5 2102.77   143.3  2103.3   175.8 2107.64   231.2  2107.9
   260.5 2104.53   286.6 2105.39   315.9 2103.77   328.9  2101.8     355 2099.93
   373.5 2096.76   377.8 2096.27   394.1 2096.92     417 2103.43   433.4 2103.72
   439.9 2105.74   449.8 2112.43   479.2 2136.62   534.9 2176.49   564.3 2195.22
   593.8 2212.21   639.6 2236.74     656 2244.22   737.8 2277.51   744.4 2279.21
#Mann= 3 ,-1 , 0
       0     .12       0   373.5    .045       0   394.1     .12       0
Bank Sta=373.5,394.1
XS Rating Curve= 0 ,0
Exp/Cntr=0.3,0.1

Type RM Length L Ch R = 1 ,14986.9 ,250.5,250,248.8
XS GIS Cut Line= 3
     2172360.459      227391.499     2172612.917      227123.763
     2172884.876      226878.618
#Sta/Elev= 30
       0 2165.87    71.6 2131.81    87.9 2125.36    97.7 2122.85   120.5 2120.38
   153.1 2118.66   169.3 2116.33   182.4 2112.65   205.2 2102.38   211.7 2100.83
     241 2100.89   263.8 2097.57   335.4 2099.28   338.7 2098.87   348.4 2095.36
   358.2 2092.86     368 2091.47   377.8 2092.84     404 2098.24   430.1 2098.82
   433.4 2099.28   436.6 2100.74     489 2136.35   531.4  2168.1   557.6 2185.14
   596.8 2209.09   626.2  2226.8     672 2251.68   698.2 2265.23   734.1  2282.3
#Mann= 3 ,-1 , 0
       0     .12       0   358.2    .045       0   377.8     .12       0
Bank Sta=358.2,377.8
XS Rating Curve= 0 ,0
Exp/Cntr=0.3,0.1

Type RM Length L Ch R = 1 ,14736.9 ,233.7,250,257.4
XS GIS Cut Line= 3
     2172517.129      227590.997     2172760.935      227318.609
     2173027.829      227064.711
#Sta/Elev= 30
       0 2136.91    22.8 2122.54    32.6 2118.12    58.8 2113.57   101.2 2110.96
   114.2 2111.54   140.4 2105.89   179.5  2106.3   202.4 2103.46     222 2104.04
   277.4 2100.55   293.8 2098.78   303.6 2094.98   323.1 2095.05   336.2 2097.16
   358.1 2092.45   365.6 2090.66   388.4  2091.9   404.7  2093.6   417.7 2097.53
   427.5 2102.35   463.4 2129.58   473.1 2138.14   502.5  2158.6   512.3 2163.44
   535.1 2178.37     597 2211.43   655.7 2237.88   704.6 2256.73   733.9 2270.63
#Mann= 3 ,-1 , 0
       0     .12       0   358.1    .045       0   388.4     .12       0
#XS Ineff= 2 , 0
          335.16 2097.18
Permanent Ineff=
       F       F
Bank Sta=358.1,388.4
XS Rating Curve= 0 ,0
Exp/Cntr=0.3,0.1

Type RM Length L Ch R = 1 ,14486.9 ,248.1,246.1,249.7
XS GIS Cut Line= 3
     2172567.024      227665.514     2172905.174      227518.688
     2173214.167       227327.84
#Sta/Elev= 30
       0 2164.91    19.6 2152.93    32.6 2141.94    45.7 2140.11    48.9 2138.64
    68.5 2124.08    97.9 2106.83   104.4    2104   215.3 2100.47   225.1 2101.77
   251.2 2098.72   270.8 2100.15   287.1 2097.35   326.2 2094.59   358.9 2087.69
   365.4 2086.92   378.5 2087.67   381.7  2088.7   388.3 2092.93   417.7 2116.26
   440.6 2131.13   463.5 2144.25   496.2 2159.67   532.2 2172.26   594.4  2188.2
   646.8 2203.48   669.7 2212.04   689.3 2214.76   705.6 2222.87   731.8 2231.68
#Mann= 3 ,-1 , 0
       0     .12       0   358.9    .045       0   378.5     .12       0
Bank Sta=358.9,378.5
XS Rating Curve= 0 ,0
Exp/Cntr=0.3,0.1

Type RM Length L Ch R = 1 ,14240.8 ,208.4,256.3,305.6
XS GIS Cut Line= 4
     2172591.626      227730.587     2172984.388      227753.899
     2173057.411      227717.388     2173400.949      227702.451
#Sta/Elev= 30
       0 2175.24    26.2 2156.31    49.2 2142.12    62.3 2129.97    75.4 2126.29
   101.6 2106.96   121.3 2097.45     141 2095.35   190.2 2094.62   216.4 2092.69
   301.6 2090.58   363.9 2091.12   393.4  2089.8     413  2087.7   419.6 2085.18
   439.2 2084.42   445.7    2085   455.5 2086.96   458.8 2088.87   517.7 2140.46
   547.1 2161.41   560.2 2163.98   573.3  2172.7   596.3 2182.48   658.5 2199.27
   684.7 2211.16   769.8 2253.68   779.7 2254.72   792.8 2262.09     819 2271.63
#Mann= 3 ,-1 , 0
       0     .12       0   419.6    .045       0   445.7     .12       0
Bank Sta=419.6,445.7
XS Rating Curve= 0 ,0
Exp/Cntr=0.3,0.1
