HEC-RAS study BACKCK2.prj: BACKCK2

--- BACKCK2.g01 (geometry) --- (continued)

Type RM Length L Ch R = 1 ,13984.4 ,303.7,290.5,273.5
XS GIS Cut Line= 3
     2172580.631      227784.044     2172949.536      227901.604
     2173215.073      228200.334
#Sta/Elev= 30
       0 2195.31    91.1 2133.88   107.4 2118.33   110.6 2116.42   123.6 2113.82
   146.4 2098.56   159.4 2093.75   224.5 2091.21   247.3 2092.44     270 2089.72
   325.4 2088.03   390.5 2087.79   403.6 2083.07   406.8 2081.64   413.4 2081.16
   429.8 2082.52   446.2 2084.92   452.7 2087.58   488.7  2114.8   508.4 2127.64
   524.8 2136.42     551  2148.5   577.2 2159.18   606.7 2169.39   619.8  2175.3
   639.4 2178.36   652.6 2183.51     682 2190.18   731.2 2198.93   786.9 2214.79
#Mann= 3 ,-1 , 0
       0     .12       0   403.6    .045       0   429.8     .12       0
Bank Sta=403.6,429.8
XS Rating Curve= 0 ,0
Exp/Cntr=0.3,0.1

Type RM Length L Ch R = 1 ,13693.9 ,189.6,201,210
XS GIS Cut Line= 3
     2172454.973      227997.861     2172808.469      228147.226
      2173113.92      228299.945
#Sta/Elev= 30
       0  2294.8    42.6 2265.64   101.7 2220.85     141 2190.12   229.6 2126.77
   265.7 2104.44   291.9 2089.85   301.8  2086.3   324.7 2083.95     328 2083.01
   334.6 2079.02   341.1 2077.17   347.7 2078.02   364.1  2077.9   383.8 2082.29
   409.8 2081.72   432.5 2083.29   448.8 2082.55   455.3  2083.8   465.1 2088.55
   491.1 2105.65   504.1 2115.13   523.6 2126.86   559.4 2144.94   604.9 2164.79
   624.4 2170.94   666.7 2181.34     696 2182.08   712.2 2186.18   725.3 2187.42
#Mann= 3 ,-1 , 0
       0     .12       0   334.6    .045       0   364.1     .12       0
Bank Sta=334.6,364.1
XS Rating Curve= 0 ,0
Exp/Cntr=0.3,0.1

Type RM Length L Ch R = 1 ,13492.9 ,258.5,245.7,240.4
XS GIS Cut Line= 4
     2172431.738      228067.565     2172670.722      228286.633
     2172730.468      228331.443     2173070.687      228326.464
#Sta/Elev= 30
       0 2284.65    26.2 2274.04    42.6 2265.79    68.8 2250.32   137.5 2203.21
     167  2181.9   245.6 2122.77   275.1 2101.77   291.4 2091.49   301.3 2086.67
   307.8 2084.59   320.9 2082.55   324.2  2080.8   330.7 2074.45   333.9 2072.77
   337.2 2072.51   356.7 2073.39   376.2 2076.75   405.4 2078.45   418.5 2080.38
   487.2 2081.07     497 2082.04   510.1 2087.54   536.3 2102.28   608.3 2138.31
   654.1 2158.27   673.7 2165.07   693.3 2169.52   706.4 2171.66   739.1 2174.29
#Mann= 3 ,-1 , 0
       0     .12       0   330.7    .045       0   356.7     .12       0
Bank Sta=330.7,356.7
XS Rating Curve= 0 ,0
Exp/Cntr=0.3,0.1

Type RM Length L Ch R = 1 ,13247.2 ,289.6,260.3,228.7
XS GIS Cut Line= 4
     2172220.968      228538.894     2172597.699      228504.042
     2172655.786      228538.894      2173015.92      228608.597
#Sta/Elev= 30
       0 2287.72      75 2248.56   117.4 2232.88   130.5 2225.35   140.2  2224.7
   146.8 2222.29   159.8 2213.01   189.2 2197.64   205.5 2187.49   296.8 2115.31
   329.4 2091.79     349 2082.89   378.3 2081.01   397.7 2069.38   410.6 2067.95
   420.3 2069.53   433.2 2073.95   439.6 2074.75     469 2077.07   544.3 2079.76
   554.2 2083.49     564 2090.44   577.1 2091.15   586.9 2096.99   606.6 2100.52
     636 2103.04     659 2108.96  713.822127.668  756.76 2145.88   812.9 2170.44
#Mann= 5 ,-1 , 0
       0     .12       0   397.7    .045       0   420.3     .12       0
  713.82    .016       0  756.76     .12       0
Bank Sta=397.7,420.3
XS Rating Curve= 0 ,0
Exp/Cntr=0.3,0.1

Type RM Length L Ch R = 1 ,12986.9 ,264.9,250,233
XS GIS Cut Line= 3
     2172292.408      228894.228     2172617.575      228749.662
     2173012.496      228635.886
#Sta/Elev= 30
       0 2301.96    22.8 2286.01    55.5 2267.23    68.6 2257.24    81.6  2255.2
    97.9  2245.7   146.9 2225.68   163.2 2217.41   189.4 2200.05   231.8 2169.85
   267.7 2141.83   277.5 2132.18   313.4 2088.59     333 2072.26   346.1 2065.09
   355.8 2063.94   365.6 2065.32     382 2072.39     395 2074.48   496.1 2074.21
   525.5 2087.75   541.8 2088.32   548.3 2090.59   577.7 2094.67   603.8 2100.32
   620.1 2105.24   646.2 2114.46  684.012132.392  721.42 2151.48   766.8 2172.49
#Mann= 5 ,-1 , 0
       0     .12       0   346.1    .045       0   365.6     .12       0
  684.01    .016       0  721.42     .12       0
Bank Sta=346.1,365.6
XS Rating Curve= 0 ,0
Exp/Cntr=0.3,0.1

Type RM Length L Ch R = 1 ,12736.9 ,276.4,292.6,302.4
XS GIS Cut Line= 3
     2172524.956       229201.74     2172774.579       228938.25
     2173052.434      228694.064
#Sta/Elev= 30
       0 2272.41    22.9 2258.67      36 2247.97    45.8 2246.58    52.3 2243.53
    71.9 2227.31   150.4 2175.87   232.2 2124.42   268.1    2099     291 2083.97
   304.1 2077.77   333.5 2070.86   349.9 2063.23   359.7 2061.75   369.5 2061.82
     376 2063.47   385.9    2067     399 2069.46   448.1 2069.66   454.6 2071.11
   467.7 2076.54   484.1 2077.11   503.7 2081.54   526.6  2089.2   549.6 2095.14
   569.2 2102.13   582.3 2107.96  606.732121.205  643.722140.954   732.9 2187.53
#Mann= 5 ,-1 , 0
       0     .12       0   349.9    .045       0     376     .12       0
  606.73    .016       0  643.72     .12       0
Bank Sta=349.9,376
XS Rating Curve= 0 ,0
Exp/Cntr=0.3,0.1

Type RM Length L Ch R = 1 ,12444.3 ,190.5,207.4,225.4
XS GIS Cut Line= 3
     2172580.045      229303.108     2172977.557      229128.881
     2173287.075      228962.345
#Sta/Elev= 30
       0 2259.19    29.4 2243.25    45.7 2231.66      62 2227.81    78.3 2216.58
   218.6 2131.98     297 2081.34   316.5 2070.11   332.8 2066.01   378.5 2066.67
   391.6  2064.2   417.7 2063.86   430.8 2060.93   443.8 2058.06   452.6 2060.83
   463.3 2067.19   473.1 2075.58   492.6 2072.88   515.4 2077.88   534.9 2073.89
  547.872074.235   587.82080.827     613 2089.74   655.3 2096.37   668.3 2096.74
   687.9 2093.83   700.9 2095.88   723.7  2106.2   762.7 2127.95   785.5 2137.69
#Mann= 5 ,-1 , 0
       0     .12       0   430.8    .045       0   452.6     .12       0
  547.87    .016       0   587.8     .12       0
Bank Sta=430.8,452.6
XS Rating Curve= 0 ,0
Exp/Cntr=0.3,0.1

Type RM Length L Ch R = 1 ,12236.9 ,253.6,250,246.2
XS GIS Cut Line= 3
     2172585.299      229323.793     2172945.943      229322.856
     2173329.225      229318.942
#Sta/Elev= 30
       0    2268      59 2240.07    72.1 2233.14      82 2225.59   101.6  2220.3
   121.3 2206.38   144.3 2192.74   183.6 2167.49   213.1 2150.74   268.8  2122.2
   291.8 2108.52   308.2 2097.35   314.8 2091.38   327.9 2078.26   334.4 2068.82
   344.2 2057.54   347.5 2055.53   350.8  2055.2   370.5 2056.65   393.4 2060.92
   406.5 2061.96   416.3 2061.43   426.2 2063.82   491.7 2064.31   534.3 2067.42
  592.842078.637   606.4 2081.39  624.542089.606   681.7 2123.39     744 2157.43
#Mann= 5 ,-1 , 0
       0     .12       0   344.2    .045       0   370.5     .12       0
  592.84    .016       0  624.54     .12       0
Bank Sta=344.2,370.5
XS Rating Curve= 0 ,0
Exp/Cntr=0.3,0.1

Type RM Length L Ch R = 1 ,11986.9 ,256.8,250,240.2
XS GIS Cut Line= 3
     2172634.198      229603.328     2172995.928      229563.136
     2173358.403      229527.246
#Sta/Elev= 30
       0 2320.25    68.9 2275.85   131.2 2233.13   183.6 2195.38   190.2 2189.93
     200 2179.84   213.1 2176.96   216.4  2174.9   242.6 2151.68   295.1 2114.19
   314.8 2098.85   324.6 2089.31   337.7 2074.46   350.8 2056.37   354.1 2053.29
   357.4 2051.84   367.2 2051.02   380.2 2053.12     390 2056.52   412.7 2060.09
   484.3 2060.61   539.6  2063.1   555.8 2064.18  563.562067.238   581.8 2075.85
   595.22084.448   611.1 2095.39   627.4 2105.02   682.7 2131.02   728.2 2154.54
#Mann= 5 ,-1 , 0
       0     .12       0   354.1    .045       0   380.2     .12       0
  563.56    .016       0   595.2     .12       0
Bank Sta=354.1,380.2
XS Rating Curve= 0 ,0
Exp/Cntr=0.3,0.1

Type RM Length L Ch R = 1 ,11736.9 ,257.6,250,246
XS GIS Cut Line= 3
     2172712.189      229908.965      2173060.07      229803.436
     2173403.277      229676.661
#Sta/Elev= 30
       0 2294.16    16.4 2283.18    85.2 2233.04   127.7 2200.91   157.2  2180.7
     190 2156.69   203.1 2144.22   216.2 2142.47   219.4 2141.19   235.8 2127.02
   268.6 2106.94   275.1 2101.94   278.4 2099.89   288.2 2097.05   301.3 2088.34
   314.4 2082.33   327.5 2073.72   340.6 2063.48   353.7 2050.45     356  2049.6
   363.5 2048.18   379.9 2050.05   412.5 2057.82   445.2 2056.67   474.6 2057.06
   487.7  2060.9  522.982082.448  555.892099.635   673.9 2156.92   729.4 2182.23
#Mann= 5 ,-1 , 0
       0     .12       0     356    .045       0   379.9     .12       0
  522.98    .016       0  555.89     .12       0
Bank Sta=356,379.9
XS Rating Curve= 0 ,0
Exp/Cntr=0.3,0.1

Type RM Length L Ch R = 1 ,11486.9 ,251.2,250,240.3
XS GIS Cut Line= 3
     2172828.708      230211.136     2173147.296      230035.364
     2173474.545      229874.172
#Sta/Elev= 30
       0  2263.6    32.8    2245      82 2212.43   173.7 2144.56     200 2126.05
   206.5 2121.05   219.6 2107.56   222.9 2105.87   232.7 2105.08     236 2103.76
   252.4  2089.5   285.2 2070.83     295 2067.22   301.6 2065.92   314.7 2059.66
   324.5  2057.6     354 2046.83   367.1 2045.86   380.2 2047.37   396.4 2051.14
   412.7 2052.64   435.5 2052.28   445.3 2053.35   461.6 2062.04  499.942090.759
  537.472116.396   591.9 2151.32   608.1 2162.89   702.6 2224.46   728.6 2240.52
#Mann= 5 ,-1 , 0
       0     .12       0     354    .045       0   380.2     .12       0
  499.94    .016       0  537.47     .12       0
Bank Sta=354,380.2
XS Rating Curve= 0 ,0
Exp/Cntr=0.3,0.1

Type RM Length L Ch R = 1 ,11236.9 ,201.8,219.2,243.2
XS GIS Cut Line= 3
     2172962.176      230435.127     2173279.961      230246.271
     2173553.883      230008.078
#Sta/Elev= 30
       0 2090.98    19.6 2094.86    32.7 2098.69    81.8 2119.31   101.4  2122.6
   117.8 2122.73   130.9 2119.53   153.8 2109.86   209.4  2081.2   222.4 2073.71
     229 2068.22   245.4 2065.86   255.2 2059.55   274.8 2051.43   284.6 2049.39
   323.9 2049.98   356.6 2044.03   366.4 2042.73   382.8 2044.38   395.8 2047.68
   405.6 2053.77   418.7 2054.57     422 2055.92   435.1  2068.2   468.62091.167
   490.7 2105.01  509.82 2118.32     579 2164.29   709.8 2243.58   732.7 2258.71
#Mann= 5 ,-1 , 0
       0     .12       0   356.6    .045       0   382.8     .12       0
   468.6    .016       0  509.82     .12       0
Bank Sta=356.6,382.8
XS Rating Curve= 0 ,0
Exp/Cntr=0.3,0.1

Type RM Length L Ch R = 1 ,11017.7 ,280.8,280.8,280.3
XS GIS Cut Line= 3
     2173027.538      230706.341     2173268.181      230454.081
     2173712.318      230420.931
#Sta/Elev= 30
       0 2190.37    45.6 2172.91    65.2 2163.95    81.5 2157.71   136.8 2131.63
   179.2 2112.89     215 2095.62   237.8 2085.89   267.2 2069.58   283.5 2057.56
     290  2054.2     303 2052.44     316  2047.7   342.1 2045.77   368.3 2047.17
   384.6 2047.02   404.3 2045.49   417.4 2041.35   420.7 2040.42   430.5 2040.01
   440.3 2041.38   453.4 2046.24   479.6  2054.2   499.3 2054.02   522.2  2060.5
   577.9  2086.1  596.622095.475  642.792119.969   712.1 2158.79     794 2201.72
#Mann= 5 ,-1 , 0
       0     .12       0   417.4    .045       0   440.3     .12       0
  596.62    .016       0  642.79     .12       0
Bank Sta=417.4,440.3
XS Rating Curve= 0 ,0
Exp/Cntr=0.3,0.1

Type RM Length L Ch R = 1 ,10736.9 ,217.8,212.8,207.8
XS GIS Cut Line= 3
     2173037.674      230748.117     2173400.545      230719.469
     2173763.416      230690.821
#Sta/Elev= 30
       0 2214.42    49.2 2210.75    72.1 2206.45   101.7 2197.14   137.7 2180.48
   170.5 2161.24   186.9 2150.14   209.9 2129.88   311.5 2052.17   324.6 2045.02
   337.8 2040.79   347.6 2036.47     364 2035.39   377.1 2035.91   393.5  2038.3
   406.6 2042.05   429.6 2042.55   449.3 2044.83   462.4 2050.56     482 2061.24
   544.4 2097.47  563.532107.726  594.792122.814   603.4 2126.19   616.5 2133.94
   623.1 2136.19   632.9 2141.43   665.7 2160.71   685.4 2171.26     728 2197.45
#Mann= 5 ,-1 , 0
       0     .12       0   347.6    .045       0   377.1     .12       0
  563.53    .016       0  594.79     .12       0
Bank Sta=347.6,377.1
XS Rating Curve= 0 ,0
Exp/Cntr=0.3,0.1

Type RM Length L Ch R = 1 ,10524.1 ,330.9,296.6,259
XS GIS Cut Line= 3
     2173077.326      231159.414     2173389.332      230938.686
     2173790.957      230852.387
#Sta/Elev= 30
       0 2268.57      49 2250.42    84.9 2234.49   104.5 2224.96   160.1 2194.98
   258.1 2134.81   267.9 2128.01   326.7 2082.29   336.5 2073.41     343  2066.1
   349.5 2060.11   359.3 2052.72   385.4 2040.83   408.3 2033.73     418 2032.79
   434.4 2034.24   457.2 2039.46   528.9 2041.73   545.2 2047.18   558.2 2054.21
  608.592076.166   640.22092.721   669.1 2108.74   682.1 2117.62   691.9 2121.01
   698.4 2125.66   737.6 2145.55   763.6  2156.6   776.7 2160.75     793 2164.51
#Mann= 5 ,-1 , 0
       0     .12       0   408.3    .045       0   434.4     .12       0
  608.59    .016       0   640.2     .12       0
Bank Sta=408.3,434.4
XS Rating Curve= 0 ,0
Exp/Cntr=0.3,0.1

Type RM Length L Ch R = 1 ,10227.5 ,270.3,264.9,261.9
XS GIS Cut Line= 4
     2173225.031      231385.121     2173474.258        231229.8
     2173497.207      231164.393     2173797.596      230855.706
#Sta/Elev= 30
       0 2233.97    65.3 2183.97    94.6 2162.67   146.8 2126.99   172.9 2110.15
   208.8 2088.57   264.3 2058.85   274.1 2052.44   277.4 2051.08   287.1 2050.35
   296.8 2044.98   306.3 2042.67   312.6 2038.71     322    2031   328.3  2029.9
   344.1 2030.67   359.8 2035.76     376 2036.16   405.4 2040.12   457.6 2044.05
   522.9 2051.71  538.352051.659   555.5 2051.95   568.6 2054.84  580.642056.083
   607.7 2058.65     624 2063.83     673 2091.44     735 2131.25   793.7    2163
#Mann= 5 ,-1 , 0
       0     .12       0     322    .045       0   344.1     .12       0
  538.35    .016       0  580.64     .12       0
Bank Sta=322,344.1
XS Rating Curve= 0 ,0
Exp/Cntr=0.3,0.1

Type RM Length L Ch R = 1 ,9962.6  ,213.6,225.7,231.4
XS GIS Cut Line= 3
     2173550.629      231588.843     2173719.594      231313.758
     2173865.815      230919.519
#Sta/Elev= 30
       0 2192.99    29.4 2175.38    94.6 2132.89   127.2 2109.45   182.6 2066.51
   215.2 2044.62   234.8 2036.42   257.6 2032.73  281.22 2031.69  327.382031.613
   339.1 2031.59   368.5 2028.36   378.2 2026.82   397.8 2028.24   407.6 2033.43
   433.7 2034.93   446.7 2039.46   492.3  2067.2   521.7  2087.8     538 2101.28
   557.5  2114.9   580.3    2126   596.6 2126.41   619.4  2121.6     639 2115.62
   687.9 2095.87   710.7 2084.56     714  2084.4   717.2 2086.19   743.3  2108.3
#Mann= 5 ,-1 , 0
       0     .12       0  281.22    .016       0  327.38     .12       0
   368.5    .045       0   397.8     .12       0
#XS Ineff= 2 , 0
          336.12 2031.79
Permanent Ineff=
       F       F
Bank Sta=368.5,397.8
XS Rating Curve= 0 ,0
Exp/Cntr=0.3,0.1

Type RM Length L Ch R = 1 ,9736.9  ,227.1,219.3,215.8
XS GIS Cut Line= 3
     2173700.158      231681.662     2173914.672      231390.536
     2174098.965      231061.109
#Sta/Elev= 30
       0 2192.47    65.2 2149.54   107.5 2118.84   169.4  2071.4     202 2048.68
   211.8 2043.63  227.632041.208  277.222034.034     303 2031.06   309.5 2029.24
   332.3 2028.75   348.6 2025.16   361.6 2023.47   374.6 2024.66   381.2 2028.03
   400.7 2034.53   413.7 2040.88   449.5 2064.02   472.3 2082.07     495 2098.69
   508.1 2109.96   524.3  2122.1   573.1 2164.81   608.9 2193.33     648 2220.03
   664.2 2227.18   677.3 2230.78   690.3 2233.01   706.6 2233.09   739.1  2228.4
#Mann= 5 ,-1 , 0
       0     .12       0  227.63    .016       0  277.22     .12       0
   348.6    .045       0   374.6     .12       0
Bank Sta=348.6,374.6
XS Rating Curve= 0 ,0
Exp/Cntr=0.3,0.1

Type RM Length L Ch R = 1 ,9517.6  ,275.2,329.7,376.6
XS GIS Cut Line= 3
      2173755.69      231716.916     2174072.844      231561.772
     2174262.792      231137.216
#Sta/Elev= 30
       0 2171.61    98.1 2110.71   107.9 2105.97   179.8  2085.3   222.3 2078.16
   248.4 2071.77   294.2 2057.37  316.072048.638   343.3 2037.96  364.11 2027.74
     376 2025.92   428.4 2027.23   441.5 2023.76   451.3 2023.44   474.3  2021.3
   480.8 2022.73   487.4 2028.65   493.9 2038.37     507 2053.98     543 2088.22
   579.1 2119.26   677.3 2198.29   719.9 2235.74   736.3  2256.7   742.8 2268.64
   755.9 2283.73   772.3 2291.78   785.4  2294.7   801.8 2295.28   818.2 2292.73
#Mann= 5 ,-1 , 0
       0     .12       0  316.07    .016       0  364.11     .12       0
   451.3    .045       0   480.8     .12       0
#XS Ineff= 2 , 0
          427.99 2027.22
Permanent Ineff=
       F       F
Bank Sta=451.3,480.8
XS Rating Curve= 0 ,0
Exp/Cntr=0.3,0.1

Type RM Length L Ch R = 1 ,9187.9  ,211.4,213.2,221.8
XS GIS Cut Line= 4
     2173787.924      231769.869     2174182.219      231674.619
     2174300.457      231705.425     2174622.304      231571.123
#Sta/Elev= 30
       0 2142.54    19.6 2137.02      72  2133.6    94.9    2128   127.6 2113.82
   189.7 2082.11   215.9 2070.66   242.1 2061.92   310.8 2044.75   353.3 2024.63
   366.4 2022.53   392.6 2024.98  412.252024.293   463.5 2021.99  477.662019.975
   479.6 2019.66   495.7 2017.74   505.3 2018.07   508.5  2019.7   511.8 2023.56
   521.4 2039.54   527.8 2046.85   534.3 2051.77   599.5 2087.64   628.9 2098.69
   677.8 2112.74   726.6 2122.32   762.5 2126.92   830.9 2128.98   876.6 2141.18
#Mann= 5 ,-1 , 0
       0     .12       0  412.25    .016       0  477.66     .12       0
   479.6    .045       0   508.5     .12       0
Bank Sta=479.6,508.5
XS Rating Curve= 0 ,0
Exp/Cntr=0.3,0.1

Type RM Length L Ch R = 1 ,8974.7  ,301.7,238.1,174
XS GIS Cut Line= 4
     2173819.553      231953.601     2174098.367      231857.344
     2174204.582      231892.196     2174633.608      231636.424
#Sta/Elev= 30
       0 2232.88    29.5 2216.93    88.5 2176.76   121.3 2151.69   203.2 2085.23
   249.1 2052.21   304.5 2021.32   314.1 2019.04   333.3 2019.18   339.7  2017.9
   349.3  2015.9   358.8 2015.51   384.4 2017.62   400.4 2021.57   426.3 2020.99
   436.1 2022.27   445.9 2026.66   455.7 2034.52   494.9 2059.14  522.082071.296
  563.552089.624   628.7 2123.43   638.5  2127.2   667.9 2142.56   700.6 2155.72
   720.2 2161.39   782.2 2170.04   837.7 2172.43   889.9 2173.04   906.2 2174.42
#Mann= 5 ,-1 , 0
       0     .12       0   339.7    .045       0   384.4     .12       0
  522.08    .016       0  563.55     .12       0
Bank Sta=339.7,384.4
XS Rating Curve= 0 ,0
Exp/Cntr=0.3,0.1

Type RM Length L Ch R = 1 ,8736.6  ,326.9,342.7,357.3
XS GIS Cut Line= 3
     2174136.156      232327.778      2174202.54      231984.239
     2174649.793      231657.205
#Sta/Elev= 30
       0 2163.72     9.8 2164.85    22.9 2163.54    39.2  2159.1    78.5 2144.64
   107.9 2129.58   140.6 2109.66   215.8 2058.89   232.2 2044.55   258.3 2016.22
   274.7 2012.58   281.2 2012.95     291 2016.34   317.2 2015.54   330.3 2019.03
   349.9 2019.64   454.8  2018.9   461.4 2020.93   477.8 2029.68   490.9 2040.88
  520.782060.397  562.072087.094   589.2  2103.9   615.4  2122.4   664.6  2154.3
   694.1 2170.38   726.9 2182.16   746.6 2187.22   766.3 2188.39     904 2187.43
#Mann= 5 ,-1 , 0
       0     .12       0   258.3    .045       0     291     .12       0
  520.78    .016       0  562.07     .12       0
Bank Sta=258.3,291
XS Rating Curve= 0 ,0
Exp/Cntr=0.3,0.1

Type RM Length L Ch R = 1 ,8393.9  ,193,182,171.6
XS GIS Cut Line= 2
     2174247.349      232326.118     2174683.826       231683.85
#Sta/Elev= 30
       0 2104.83    13.1 2103.94      36  2095.9     118 2055.79   144.2 2044.83
   163.8 2038.48     190 2034.67   275.2 2030.09   304.7 2027.08   324.4 2022.75
   340.8 2017.05  357.532014.652     367 2014.96   376.8 2013.88   386.6 2012.09
   399.7 2008.21   412.8 2005.76     426 2006.59   429.2 2008.13   455.4 2045.57
   468.6 2060.76   481.6 2073.24     521 2105.11   570.1 2135.14   635.6 2169.48
   707.7  2196.6   727.4 2202.61   740.5  2205.1   756.9 2205.95   776.5 2202.86
#Mann= 4 ,-1 , 0
       0     .12       0  357.53    .016       0   399.7    .045       0
   429.2     .12       0
Bank Sta=399.7,429.2
XS Rating Curve= 0 ,0
Exp/Cntr=0.3,0.1

Type RM Length L Ch R = 1 ,8212    ,226.3,247.1,265.8
XS GIS Cut Line= 3
      2174544.96      232397.691       2174650.3      232039.909
      2174769.08       231694.33
#Sta/Elev= 30
       0 2094.15   111.2 2064.59   170.1 2045.63   176.7 2044.23   206.1    2035
   225.7 2029.76   251.9 2021.34  261.122016.965   268.3 2014.56   287.9    2012
   298.22011.564     337 2012.31   346.8 2010.51   363.2 2003.21   366.4  2002.3
     386 2001.96   399.1 2002.45   402.3 2005.59   405.6 2012.17   412.1 2026.75
   418.6 2037.49   425.2 2047.12   428.4 2050.96   431.7 2053.43   493.7 2079.63
   539.4 2097.05   581.8 2116.04   643.8 2151.27   656.8 2159.33   738.4 2201.45
#Mann= 5 ,-1 , 0
       0     .12       0  261.12    .016       0   298.2     .12       0
   363.2    .045       0   399.1     .12       0
Bank Sta=363.2,399.1
XS Rating Curve= 0 ,0
Exp/Cntr=0.3,0.1

Type RM Length L Ch R = 1 ,7964.9  ,233.5,235,236.5
XS GIS Cut Line= 2
     2174570.342      232414.062     2175113.052      231925.526
#Sta/Elev= 30
       0 2110.53    62.2 2106.48    85.1 2103.02   104.8 2096.81   147.4  2079.1
   170.3 2067.38   189.9 2056.46   229.2 2031.74   265.2 2011.84  279.432010.504
   291.4 2009.56  312.662010.079   327.4 2010.36   347.1 2007.89   353.6 2006.08
   363.5 2000.88     370 1998.16   379.8 1997.04   386.4  1997.5   396.2 2001.16
   412.6 2012.59   419.1 2015.11   451.9 2022.15   484.6 2030.99   569.8 2045.87
   651.6 2057.92   674.5 2067.16   697.5 2081.53   707.3 2085.48   730.2 2099.62
#Mann= 5 ,-1 , 0
       0     .12       0  279.43    .016       0  312.66     .12       0
   363.5    .045       0   396.2     .12       0
Bank Sta=363.5,396.2
XS Rating Curve= 0 ,0
Exp/Cntr=0.3,0.1

Type RM Length L Ch R = 1 ,7729.9  ,257.5,263.6,269.6
XS GIS Cut Line= 2
     2174717.554      232577.637      2175279.49      232110.367
#Sta/Elev= 30
       0 2163.38    32.8 2141.89   124.5  2078.2   196.6 2031.25     236 2009.41
   239.2 2008.44   249.1 2008.17  255.472006.614   268.7 2004.71   296.32004.994
   317.9  2004.8   344.1 2002.51   357.2 1998.61   363.8 1996.55   370.3 1996.06
   383.4 1996.75     390 1999.26   412.9  2009.5     426 2013.81   442.4 2017.45
   452.3 2018.61   511.2 2031.56   530.9  2033.8   553.9 2037.89     567 2041.36
   586.6 2044.71   596.5 2047.69   619.4 2057.78   681.7 2091.58   730.8 2115.66
#Mann= 5 ,-1 , 0
       0     .12       0  255.47    .016       0   296.3     .12       0
   357.2    .045       0     390     .12       0
Bank Sta=357.2,390
XS Rating Curve= 0 ,0
Exp/Cntr=0.3,0.1

Type RM Length L Ch R = 1 ,7466.3  ,259.8,219.8,185
XS GIS Cut Line= 3
     2174789.858      232761.424      2175145.76      232551.355
      2175385.67      232267.335
#Sta/Elev= 30
       0  2208.4    49.2 2173.58     187 2094.04   239.4  2060.9  274.362035.844
   288.6 2020.26   291.9 2018.46     305 2016.68  314.412008.979     328 1996.45
   331.3 1994.98   337.8 1995.06   354.2 1993.75   367.4 1996.32   377.2 1998.27
   396.9 1999.59   452.4 1999.81   494.8 2001.35   514.4 2007.29   527.4 2010.09
   543.7 2012.56   599.2 2018.06     635 2025.15   654.6 2032.88   674.2 2043.15
   719.8 2071.51   726.4 2076.39   736.1 2081.72   755.7  2095.1   785.1 2112.52
#Mann= 5 ,-1 , 0
       0     .12       0  274.36    .016       0  314.41     .12       0
   337.8    .045       0   367.4     .12       0
Bank Sta=337.8,367.4
XS Rating Curve= 0 ,0
Exp/Cntr=0.3,0.1

Type RM Length L Ch R = 1 ,7246.5  ,233.2,252.9,264.9
XS GIS Cut Line= 4
     2175105.366      232989.961     2175294.562      232694.551
     2175292.902       232616.55     2175442.276      232301.859
#Sta/Elev= 30
       0 2167.59    36.1 2153.82    65.6 2138.28    91.8 2122.78   114.8 2108.23
   147.5 2083.97   193.4 2053.14  242.192022.692     259 2012.95   268.8 2005.58
   275.4 2003.54  282.592003.352   288.5 2003.18   298.4 2000.18   304.9 1999.28
   334.4 1996.33   350.8 1995.76   383.3 1992.02   402.8 1990.55   412.6 1991.76
   422.3  1999.4   425.6 2000.84   441.8 2004.05     507 2013.53   542.8 2021.33
   575.3 2022.62   591.6 2026.71   669.7 2057.29     712 2080.61   777.2 2119.81
#Mann= 5 ,-1 , 0
       0     .12       0  242.19    .016       0  282.59     .12       0
   383.3    .045       0   412.6     .12       0
Bank Sta=383.3,412.6
XS Rating Curve= 0 ,0
Exp/Cntr=0.3,0.1

Type RM Length L Ch R = 1 ,6993.6  ,194.5,243.6,294.2
XS GIS Cut Line= 4
     2175182.962      233026.593     2175516.949      232750.978
     2175548.362      232684.625     2175774.188      232540.208
#Sta/Elev= 30
       0  2169.3    65.6 2122.05   147.6  2060.2     187 2032.66     210 2018.68
   223.1 2012.02   232.9 2008.07  250.552003.107   272.3 2003.06  293.611997.078
   308.4  1995.6   360.8 1995.88   390.4 1994.24   413.3 1995.08   439.4 1991.59
   458.2  1987.8   474.5 1986.61   480.9 1987.88   487.3 1993.74   496.9 2007.78
     500 2011.09   506.4  2014.9   522.8 2021.31   565.3  2045.9   601.2 2063.88
   617.6 2070.74   653.5 2082.41   673.2 2091.77     696  2104.6   774.5 2153.94
#Mann= 5 ,-1 , 0
       0     .12       0  250.55    .016       0  293.61     .12       0
   458.2    .045       0   480.9     .12       0
Bank Sta=458.2,480.9
XS Rating Curve= 0 ,0
Exp/Cntr=0.3,0.1

Type RM Length L Ch R = 1 ,6750    ,250.8,221.5,189.3
XS GIS Cut Line= 3
     2175212.379      233079.036     2175580.014      232892.044
     2175983.184      232982.658
#Sta/Elev= 30
       0 2178.18    22.9 2165.06   170.2 2054.45   199.7 2034.17   229.1 2016.92
   245.5 2008.32   255.3 2005.29   281.5 2001.09  316.51 2001.03   324.1 2000.25
   343.7 1993.61  364.621993.851   428.9 1990.49   458.4 1986.67     478 1985.42
   491.2 1986.85     501  1990.8   510.8 1992.15   569.9 1992.51   602.7 2008.02
     642 2029.41   651.9  2033.1   687.9 2037.47   737.1 2029.34   743.7 2029.62
   756.8 2035.73   779.8 2053.01   799.4 2063.68   815.8 2077.66   825.7 2083.18
#Mann= 5 ,-1 , 0
       0     .12       0  316.51    .016       0  364.62     .12       0
   458.4    .045       0   491.2     .12       0
Bank Sta=458.4,491.2
XS Rating Curve= 0 ,0
Exp/Cntr=0.3,0.1

Type RM Length L Ch R = 1 ,6528.5  ,281.4,277,270.9
XS GIS Cut Line= 3
     2175285.662      233263.305      2175625.94      233061.916
     2175992.762      233043.838
#Sta/Elev= 30
       0 2203.43    62.1 2162.56   101.3 2132.05   218.9 2045.83   248.4 2026.43
   277.8 2009.59   297.4 2002.46   310.4 2001.73   313.7 2000.27     317  1997.3
   320.2 1993.29   326.8 1982.75   327.5 1982.16     330 1980.07   333.3 1979.65
   352.9 1981.83   372.5 1986.86   415.1 1990.39  432.051989.645   444.6 1990.26
  485.811989.722   513.5 1991.51   552.8 1995.74   575.8 1997.16   585.6    1999
   644.6 2028.74     661 2038.01   674.1 2041.76   687.2 2050.55   762.7 2088.56
#Mann= 5 ,-1 , 0
       0     .12       0   327.5    .045       0   352.9     .12       0
  432.05    .016       0  485.81     .12       0
Bank Sta=327.5,352.9
XS Rating Curve= 0 ,0
Exp/Cntr=0.3,0.1

Type RM Length L Ch R = 1 ,6251.5  ,267.9,264.7,261.5
XS GIS Cut Line= 3
     2175317.414      233339.603     2175684.187      233344.582
      2176017.05      233096.475
#Sta/Elev= 30
       0 2192.05      36 2171.75    91.7 2137.23   121.2 2117.06   134.3 2106.49
   183.4 2074.72   248.9 2036.44   275.1  2025.1   317.7 2016.28   330.8  2010.7
   343.9 2002.32   360.3 2001.22   366.8 1997.58   386.4 1982.45   396.2  1979.1
   409.3 1977.36   419.1 1977.84   422.4 1979.48   428.9 1984.17   435.4 1985.36
   471.4 1984.86  485.431986.117  524.011986.642   553.1 1986.16   566.2 1990.58
   582.6    1993   595.6 1998.75   615.2 2001.58   638.1 2008.28     782 2089.33
#Mann= 5 ,-1 , 0
       0     .12       0   396.2    .045       0   422.4     .12       0
  485.43    .016       0  524.01     .12       0
Bank Sta=396.2,422.4
XS Rating Curve= 0 ,0
Exp/Cntr=0.3,0.1

Type RM Length L Ch R = 1 ,5986.9  ,282,264.1,245.4
XS GIS Cut Line= 3
     2175629.783      233747.809     2175898.888      233498.655
     2176168.816      233253.234
#Sta/Elev= 30
       0 2172.51    29.5 2151.96    75.3 2118.51   180.1 2038.98   206.3 2020.15
   225.9  2007.7     239  2000.9     262 1993.33   281.6 1984.35   288.2 1983.18
  323.711983.853     334 1983.09   353.6 1978.34   366.7 1974.79   376.5 1975.44
     383 1977.74     396 1981.61   412.3 1985.08     471 1991.66     484 1996.66
   529.6 2011.16   545.9 2014.97   607.8 2026.94   617.6 2027.65   627.3 2022.88
   633.8 2022.34   640.4 2024.41   679.4 2043.19   705.5  2050.1   731.6  2055.5
#Mann= 4 ,-1 , 0
       0     .12       0  323.71    .016       0   353.6    .045       0
     383     .12       0
Bank Sta=353.6,383
XS Rating Curve= 0 ,0
Exp/Cntr=0.3,0.1

Type RM Length L Ch R = 1 ,5722.8  ,190.4,179.8,168.1
XS GIS Cut Line= 3
     2175837.301      233937.081     2176079.556      233710.231
      2176225.17      233299.049
#Sta/Elev= 30
       0 2158.47    48.8 2126.02   133.4 2066.79   165.9 2046.14   188.7 2032.92
     218 2017.94   250.5 2004.43   270.1 2000.07   296.1 1997.22   302.6 1995.16
  307.821991.726   325.4 1980.58   328.6 1979.33     345 1978.92   351.21976.425
   351.6 1976.23   361.4 1974.65   384.4 1976.06     404 1979.72     427 1981.72
   456.5 1986.21   499.2 1990.18   541.8 1992.39   587.7 2002.05   613.9 2013.11
   646.7 2031.48   686.1 2054.94   735.3 2080.99   751.7 2087.62   768.1 2092.19
#Mann= 5 ,-1 , 0
       0     .12       0  307.82    .016       0   351.2     .12       0
   351.6    .045       0   384.4     .12       0
Bank Sta=351.6,384.4
XS Rating Curve= 0 ,0
Exp/Cntr=0.3,0.1

Type RM Length L Ch R = 1 ,5543.1  ,238.9,302.3,360.2
XS GIS Cut Line= 4
     2175880.135      233978.438      2176262.08      233839.549
     2176272.496      233605.174     2176481.181      233424.778
#Sta/Elev= 30
       0 2148.88    13.1 2139.16    49.2 2115.51   173.7 2025.34   219.6 1995.92
   242.5 1987.94   268.8 1984.22   304.8 1980.84   336.21981.042  377.31 1979.44
   406.4 1978.61   422.7 1975.15     452 1977.68   487.9 1977.98   536.8 1976.47
   559.6 1973.58   569.3 1972.58   579.1 1972.68   585.6 1973.94   595.4 1977.74
   618.2 1977.82   637.8 1982.14   660.5 1985.37   683.2 1993.76   709.2 2007.93
   731.9 2021.81   835.7 2095.96   897.4 2134.72   910.4 2145.13   916.9 2147.34
#Mann= 5 ,-1 , 0
       0     .12       0   336.2    .016       0  377.31     .12       0
   559.6    .045       0   585.6     .12       0
Bank Sta=559.6,585.6
XS Rating Curve= 0 ,0
Exp/Cntr=0.3,0.1

Type RM Length L Ch R = 1 ,5240.7  ,238,260.7,282.5
XS GIS Cut Line= 4
     2175896.123      234005.096     2176287.007      233867.894
     2176408.122      233865.784     2176648.801      233764.998
#Sta/Elev= 30
       0 2143.96    48.9    2111    91.3 2078.44   166.4  2023.5   208.8 1997.18
   231.6 1989.44   264.2 1983.99   303.4 1980.28  336.641979.764  377.841979.865
   420.8 1977.35   437.2 1971.16   443.7 1969.18   450.3 1969.08   466.6 1970.48
   496.1 1973.35   512.5 1973.55   522.3 1979.09   538.7 1992.13     555 2000.38
   597.4 2011.68   626.7 2023.09   708.3 2062.62   721.3 2070.66   724.6 2071.88
   734.4  2072.5   737.6 2074.02   744.1 2079.84   747.4 2081.68   796.3 2105.18
#Mann= 5 ,-1 , 0
       0     .12       0  336.64    .016       0  377.84     .12       0
   437.2    .045       0   466.6     .12       0
Bank Sta=437.2,466.6
XS Rating Curve= 0 ,0
Exp/Cntr=0.3,0.1

Type RM Length L Ch R = 1 ,4980    ,333.5,254.5,174.5
XS GIS Cut Line= 4
     2175970.022      234246.284     2176223.942      234088.622
     2176315.899      234145.105     2176706.508      233926.968
#Sta/Elev= 30
       0 2160.77      26 2143.73      39 2136.64    71.5 2113.57    84.5 2103.89
    94.2 2093.67   110.5 2080.38   159.2 2045.01   207.9 2007.47   233.9  1989.2
   243.7 1985.66   298.9 1979.52     312 1973.66   344.7 1967.13   357.8 1966.34
   367.6 1967.24   390.4 1973.16   423.1 1974.86   429.7 1976.83   439.5 1982.16
  454.581984.219  486.641990.125   599.5 1999.78   628.9 2004.93     704 2027.26
   739.9 2044.57     753 2052.99   769.3 2055.06   785.6  2065.3   854.2 2095.54
#Mann= 5 ,-1 , 0
       0     .12       0   344.7    .045       0   367.6     .12       0
  454.58    .016       0  486.64     .12       0
Bank Sta=344.7,367.6
XS Rating Curve= 0 ,0
Exp/Cntr=0.3,0.1

Type RM Length L Ch R = 1 ,4725.6  ,295.7,305.7,315.3
XS GIS Cut Line= 3
     2176322.769      234612.811     2176336.733      234233.647
     2176727.565      233966.048
#Sta/Elev= 30
       0  2133.5    42.5 2114.59    68.7 2104.03   127.6 2076.04   222.4 2016.39
   268.2 1990.52   287.8 1974.73   294.4 1971.87   327.1 1963.92   333.6 1962.95
   346.7 1962.98   353.2 1964.08   359.8 1966.14   366.3 1970.81   372.9 1973.64
   408.8 1980.39   418.6 1981.08   444.8 1980.37   464.4 1982.84  478.091982.726
     497 1985.45  517.761991.314     595 1999.86   617.9 2004.22   686.5 2028.74
   719.2 2042.28   735.5  2050.8   748.6 2052.15   761.6 2059.33   853.1 2096.32
#Mann= 5 ,-1 , 0
       0     .12       0   327.1    .045       0   353.2     .12       0
  478.09    .016       0  517.76     .12       0
Bank Sta=327.1,353.2
XS Rating Curve= 0 ,0
Exp/Cntr=0.3,0.1

Type RM Length L Ch R = 1 ,4419.9  ,239.4,258.5,277.2
XS GIS Cut Line= 2
     2176515.552      234712.813      2176738.42      233987.385
#Sta/Elev= 30
       0 2173.07    22.9 2156.63      72  2123.1     121 2087.29   206.1 2027.09
   255.1 1991.06   287.9 1969.75   294.4  1966.6   304.2 1964.38   359.8 1965.12
   382.7 1961.19   389.3 1960.04   399.1 1959.91   412.2 1960.77   418.7 1963.49
     435 1974.75   448.1 1980.32     458 1985.84   467.8 1986.64  475.321988.568
  510.081999.361   588.8 2028.95   618.2  2038.1   631.3 2039.24   644.4 2047.68
   654.2 2051.93     664 2057.45   686.9 2068.45   716.4 2080.81   758.9 2095.07
#Mann= 5 ,-1 , 0
       0     .12       0   382.7    .045       0   412.2     .12       0
  475.32    .016       0  510.08     .12       0
#XS Ineff= 2 , 0
          359.86 1965.14
Permanent Ineff=
       F       F
Bank Sta=382.7,412.2
XS Rating Curve= 0 ,0
Exp/Cntr=0.3,0.1

Type RM Length L Ch R = 1 ,4161.5  ,177.8,175.9,175.8
XS GIS Cut Line= 3
     2176547.565      234742.507     2176856.252      234450.416
     2176884.466      234110.196
#Sta/Elev= 30
       0 2180.57    29.4  2161.4   150.4 2073.61   281.1 1973.77   287.7 1969.85
   297.5 1965.82   323.6 1961.72     340 1961.07   353.1 1958.32   366.1 1957.11
   382.5 1958.33   402.1 1961.12   411.9 1967.68   421.7 1977.48     425 1979.54
   431.5 1980.95   441.2 1985.16   470.5 1990.78   493.2 1991.08   506.3  1994.1
  538.221998.819  589.842007.885   600.6 2010.43   610.3 2014.96   629.8 2016.82
   642.8 2023.58   678.6 2033.52   707.8 2042.96   733.8 2053.35   766.4 2070.34
#Mann= 5 ,-1 , 0
       0     .12       0   353.1    .045       0   382.5     .12       0
  538.22    .016       0  589.84     .12       0
Bank Sta=353.1,382.5
XS Rating Curve= 0 ,0
Exp/Cntr=0.3,0.1

Type RM Length L Ch R = 1 ,3985.6  ,227.4,223.5,216.9
XS GIS Cut Line= 2
     2176678.674      234881.914     2177170.066      234344.758
#Sta/Elev= 30
       0 2208.54    13.1 2199.72    26.2  2189.7    45.9 2176.76   111.5 2127.34
   124.6 2114.11   147.6 2094.71   259.1  2006.2   288.6 1980.64   295.1 1973.85
   301.7 1965.71     305 1962.74   311.5 1959.24   318.7 1957.21   327.9 1955.36
   347.6  1956.6     364 1957.44   377.1 1959.88   416.5 1963.78   455.8  1966.5
     505 1977.21   521.4 1977.86  536.821981.148   554.2 1981.64     564 1985.86
  578.591988.579   616.5  1995.8   688.7 2004.55   705.1 2009.04     728  2017.9
#Mann= 5 ,-1 , 0
       0     .12       0   318.7    .045       0   347.6     .12       0
  536.82    .016       0  578.59     .12       0
Bank Sta=318.7,347.6
XS Rating Curve= 0 ,0
Exp/Cntr=0.3,0.1

Type RM Length L Ch R = 1 ,3762    ,177.9,156,130.3
XS GIS Cut Line= 3
     2176862.891      235061.152     2177164.858      234645.105
     2177221.858      234395.805
#Sta/Elev= 30
       0 2215.42    19.6 2202.55    55.7 2180.85    81.9 2161.78   104.8 2147.48
   153.9 2113.27   170.3 2101.54   180.1 2093.52   189.9 2087.06   225.9 2058.65
   242.3 2047.19   301.2  2001.6   324.2 1980.36   340.5 1961.83   347.1 1955.86
   350.4 1954.24   356.9 1953.41   373.3 1954.42   386.4 1954.86   396.2 1957.13
     406 1958.06   484.6 1958.48   504.3 1961.29  561.021965.161   607.81970.185
   632.1  1974.6     642 1977.56   674.7 1989.61   733.8 2000.85   769.8  2011.8
#Mann= 5 ,-1 , 0
       0     .12       0   347.1    .045       0   373.3     .12       0
  561.02    .016       0   607.8     .12       0
Bank Sta=347.1,373.3
XS Rating Curve= 0 ,0
Exp/Cntr=0.3,0.1

Type RM Length L Ch R = 1 ,3606    ,193.3,151.4,110.9
XS GIS Cut Line= 4
     2177004.412      235108.791     2177211.009      234874.416
     2177211.009      234643.514     2177304.759      234429.972
#Sta/Elev= 30
       0  2160.9    45.6 2130.34   123.7 2075.35   169.2 2045.45   198.5 2027.27
   247.3 2000.34   276.6 1988.55   315.7 1974.82     332 1965.84   335.2 1963.35
     345 1953.57   348.2 1951.56     358 1951.06     371 1951.17   380.7 1953.13
   393.7 1954.65   403.5 1957.17   426.3 1956.93   439.3 1958.27     475 1959.84
   484.8 1958.36   536.8 1961.75  554.491962.188  597.761968.122   627.6 1973.22
     647 1978.07   669.7 1986.27   708.5 1998.07   760.4 2015.56   776.6 2021.96
#Mann= 5 ,-1 , 0
       0     .12       0     345    .045       0   380.7     .12       0
  554.49    .016       0  597.76     .12       0
Bank Sta=345,380.7
XS Rating Curve= 0 ,0
Exp/Cntr=0.3,0.1

Type RM Length L Ch R = 1 ,3454.6  ,37.5,38.8,37.5
XS GIS Cut Line= 4
     2177220.992      235133.314     2177433.665      234829.494
     2177280.671      234734.008     2177329.065      234436.916
#Sta/Elev= 30
       0  2083.9    45.5 2057.99    87.8 2036.16   136.6 2018.85     218 1996.76
     270 1980.59   302.5 1972.72   331.8 1967.39   348.1 1965.75   370.9 1961.95
   393.8  1959.9   423.3 1952.71   436.4 1951.62   446.3 1949.79   456.1 1949.58
   462.7 1949.75   470.1 1951.68   531.5 1958.14   570.8 1958.82  591.831957.342
   603.6 1958.88   623.2  1958.9   640.11960.086   672.3 1967.03   698.4 1977.26
   711.5 1981.48     741 1988.98   786.8 2002.29   816.2  2013.9   852.2 2026.68
#Mann= 5 ,-1 , 0
       0     .12       0   436.4    .045       0   470.1     .12       0
  591.83    .016       0   640.1     .12       0
Bank Sta=436.4,470.1
XS Rating Curve= 0 ,0
Exp/Cntr=0.3,0.1

Type RM Length L Ch R = 1 ,3415.8  ,136.7,172.2,208.9
XS GIS Cut Line= 4
     2177251.374      235131.144     2177472.728      234816.474
     2177319.733      234720.988     2177367.259      234436.916
#Sta/Elev= 30
       0 2073.22    65.2 2038.81    97.8 2026.15   143.5  2013.1   182.6  2003.2
   260.8 1978.84     300  1970.7  350.17 1963.84   361.9 1961.21   378.2 1955.17
   381.5 1954.67   433.9  1954.2     447 1952.92   456.9 1950.71   463.4 1949.23
   479.8 1948.92   489.7 1950.59   499.5  1953.1   509.3 1954.29   548.7 1955.89
   594.5 1955.16   607.6  1958.1  612.791958.144   633.8 1958.12   646.9 1960.46
   663.3  1967.9   702.5 1982.38   738.5 1993.32   781.1 2009.14   853.1 2038.88
#Mann= 5 ,-1 , 0
       0     .12       0  350.17    .016       0   456.9    .045       0
   489.7    .016       0  612.79     .12       0
Bank Sta=456.9,489.7
XS Rating Curve= 0 ,0
Exp/Cntr=0.3,0.1

Type RM Length L Ch R = 1 ,3243.7  ,244.1,280.8,316.5
XS GIS Cut Line= 4
     2177317.505      235138.551     2177565.899      234860.383
     2177539.727      234648.968     2177590.075       234496.19
#Sta/Elev= 30
       0 2049.57    29.4 2038.28    58.9 2028.42   160.3 2001.26   212.6 1990.15
  307.741968.048   333.7 1958.52  349.491954.967   359.8 1954.95   395.9  1952.1
     445 1954.14   448.3 1953.37   454.9 1949.69   458.1 1949.14     468 1950.48
   487.6 1951.18   517.1 1951.51   523.7 1950.05   543.4 1948.22   555.2 1950.03
   569.6 1953.59   582.7 1960.95   598.8 1976.79   608.5  1988.1   621.4 2000.13
   637.4 2013.13   669.6  2034.1   701.8 2052.99   730.7 2066.61   746.8 2073.15
#Mann= 5 ,-1 , 0
       0     .12       0  307.74    .016       0  349.49     .12       0
   523.7    .045       0   555.2     .12       0
#XS Ineff= 2 , 0
          444.76 1954.12
Permanent Ineff=
       F       F
Bank Sta=523.7,555.2
XS Rating Curve= 0 ,0
Exp/Cntr=0.3,0.1

Type RM Length L Ch R = 1 ,2962.9  ,236.2,226,217.8
XS GIS Cut Line= 4
     2177510.213      235199.315     2177675.144      234904.176
     2177786.255      234801.746     2177817.505      234582.996
#Sta/Elev= 30
       0 2055.85      78 2011.23   100.8 1999.66   123.5 1990.07   162.6  1979.4
   208.1 1972.25  227.961967.212   237.3 1964.82  270.891960.691   282.8 1959.15
   299.1 1958.68   315.3 1955.36   334.8 1953.01   347.7 1948.98   363.8 1946.92
   428.1  1947.9   437.8 1947.63     441 1946.51   444.2 1945.08   450.6  1944.6
   463.5 1944.75   473.1 1946.49   476.4 1949.19   489.2 1964.73   508.7  1975.6
   554.2 2005.65   599.7 2028.82   671.2 2073.87   693.9 2083.37   710.2 2092.08
#Mann= 5 ,-1 , 0
       0     .12       0  227.96    .016       0  270.89     .12       0
     441    .045       0   473.1     .12       0
Bank Sta=441,473.1
XS Rating Curve= 0 ,0
Exp/Cntr=0.3,0.1

Type RM Length L Ch R = 1 ,2736.9  ,244.5,245.9,244.6
XS GIS Cut Line= 3
     2177708.634      235312.267     2177896.637       235003.41
     2178114.323      234694.713
#Sta/Elev= 30
       0 2028.61    32.6  2014.5    61.9 2003.35    97.7 1991.28   133.6 1980.66
   149.8 1971.35   175.9 1953.89   182.4 1951.28  187.161950.268   205.2 1947.48
   218.2 1947.93  227.081947.037   244.3 1944.74   257.3    1945   267.1 1943.64
   338.8 1944.97   348.6 1943.51   358.3 1942.32   368.1 1942.14   377.9 1943.83
   394.1 1944.67   403.9 1946.97   416.9 1955.24   449.5 1971.72   498.3 1999.04
   599.3 2045.58   635.1 2059.14   661.2 2070.52   687.2 2085.41   739.3 2112.66
#Mann= 5 ,-1 , 0
       0     .12       0  187.16    .016       0  227.08     .12       0
   348.6    .045       0   377.9     .12       0
Bank Sta=348.6,377.9
XS Rating Curve= 0 ,0
Exp/Cntr=0.3,0.1

Type RM Length L Ch R = 1 ,2491    ,244.5,236.2,227.5
XS GIS Cut Line= 2
     2177909.519      235418.065       2178293.2      234834.732
#Sta/Elev= 30
       0    2013    19.7  2006.1   47.441997.843   66.471992.647   154.1 1970.63
   167.2 1964.82  180.711956.224   190.1 1949.03  200.861944.426   226.2 1943.47
     236 1944.12   249.1 1943.39   268.8 1944.64   291.7 1943.03   311.4 1943.66
   321.2 1942.86   333.1 1940.18   344.2 1938.06   363.8 1939.36   367.1 1941.16
   386.8 1958.68   399.9 1969.04   419.6 1981.59   452.4 1998.35   485.1 2016.45
     554 2058.84     590 2082.65   603.1 2090.49   652.3 2117.94   698.2 2142.15
#Mann= 7 ,-1 , 0
       0     .12       0   47.44     .06       0   66.47     .12       0
  180.71    .016       0  200.86     .12       0   333.1    .045       0
   363.8     .12       0
Bank Sta=333.1,363.8
XS Rating Curve= 0 ,0
Exp/Cntr=0.3,0.1

Type RM Length L Ch R = 1 ,2254.8  ,305.3,313,320.1
XS GIS Cut Line= 4
       2178043.2      235506.607     2178268.894      235327.787
     2178357.436      235091.676     2178380.005      234878.135
#Sta/Elev= 30
       0 2010.18    32.7 2001.91   87.95  1994.1   153.8 1984.63   238.9 1965.56
   314.2 1954.28  330.651950.189   337.1 1948.19   353.4 1940.73  364.671939.769
   369.8 1939.52   379.6 1936.39   386.2 1935.08     396 1934.78   405.8 1936.42
   412.4 1938.36   425.5 1940.09   471.3 1937.49   484.4 1940.83   507.4 1940.88
   513.9 1943.56   520.5  1949.1     527 1956.32   553.1 1991.49   601.9  2036.2
   631.2 2060.53   676.8 2094.82     693 2105.72   715.8 2119.96   754.8 2140.97
#Mann= 6 ,-1 , 0
       0     .06       0   87.95     .12       0  330.65    .016       0
  364.67     .12       0   379.6    .045       0   405.8     .12       0
Bank Sta=379.6,405.8
XS Rating Curve= 0 ,0
Exp/Cntr=0.3,0.1

Type RM Length L Ch R = 1 ,1941.8  ,536,522.7,508.9
XS GIS Cut Line= 4
      2178511.95      235721.885       2178543.2      235419.801
     2178715.075       235143.76      2178636.95      234914.593
#Sta/Elev= 30
       0 2052.05    78.4  2030.7   124.1 2013.22   166.5 1994.18   248.2 1963.99
     258 1958.61     271 1957.24   280.8 1953.25   303.7 1950.18   316.7 1939.18
     320 1937.68   342.7 1936.18   355.7 1933.56     372 1932.21     385 1934.01
     398 1936.77     424 1937.07  434.671935.844   453.3 1934.42  473.561936.706
  516.961936.962   606.1 1938.54   612.6 1939.88   620.61945.292   632.1 1952.82
     655 1960.65     678 1973.78     727 2005.76   766.3 2034.37     871 2107.23
#Mann= 7 ,-1 , 0
       0     .12       0   355.7    .045       0     385     .12       0
  434.67     .06       0  473.56    .016       0  516.96     .08       0
   620.6     .12       0
#XS Ineff= 2 , 0
                          500.63         1954.21
Permanent Ineff=
       F       F
Bank Sta=355.7,385
XS Rating Curve= 0 ,0
Exp/Cntr=0.3,0.1

Type RM Length L Ch R = 1 ,1419.1  ,471,461.5,449.2
XS GIS Cut Line= 3
     2178937.731      235781.346     2179067.939      235149.836
     2179141.724      235021.798
#Sta/Elev= 30
       0 2034.01    42.6 2012.22   74.781998.458   114.6 1982.26   127.6 1972.76
   140.7 1970.15     144 1968.52   176.8 1948.17   193.1 1930.69   199.7 1927.39
     216 1926.31   232.4 1927.78   245.5 1930.01     288  1932.9   301.1 1932.22
   314.2  1929.8   350.2 1931.31   376.4 1928.98   386.2 1932.22   435.3 1934.56
  446.731936.196   464.8 1940.03  482.121941.315   540.1 1940.82   612.1 1947.11
   625.2 1950.64   654.4 1961.34   718.7 1981.81   747.6 1993.32   792.6 2015.86
#Mann= 6 ,-1 , 0
       0     .12       0   74.78     .07       0   199.7    .045       0
   232.4     .12       0  446.73    .016       0  482.12     .12       0
Bank Sta=199.7,232.4
XS Rating Curve= 0 ,0
Exp/Cntr=0.3,0.1

Type RM Length L Ch R = 1 ,957.6   ,506.9,519.3,530.2
XS GIS Cut Line= 3
      2179393.46      235813.898     2179428.182      235590.374
     2179410.821       235063.03
#Sta/Elev= 30
       0 2018.58    26.2 2006.01    55.7 1993.76   104.9 1973.96     141 1961.65
   180.3 1953.32   209.8 1948.89   239.3 1945.45   275.4 1943.23   285.2  1937.9
   298.3 1927.83   301.6 1926.72     318 1926.22   344.2 1923.39   363.8 1921.63
   383.5 1923.12  394.211925.463     413 1926.21  428.921924.592  469.381925.901
  493.46 1926.92   534.3 1927.32   573.6 1949.55   580.1 1952.09   593.2 1955.57
   662.1 1967.09   675.2 1970.25   688.3  1975.3   704.7 1983.61   753.8 2012.74
#Mann= 7 ,-1 , 0
       0     .12       0   344.2    .045       0   383.5     .12       0
  394.21    .016       0  428.92     .12       0  469.38     .08       0
  493.46     .12       0
Bank Sta=344.2,383.5
XS Rating Curve= 0 ,0
Exp/Cntr=0.3,0.1

Type RM Length L Ch R = 1 ,438.3   ,335.8,341.4,347
XS GIS Cut Line= 4
      2179688.44      235825.805      2179728.37      235745.944
     2179851.359      235186.728     2179827.488      235047.839
#Sta/Elev= 30
       0 1979.54    22.3 1966.76    55.51949.917    76.5  1944.4    95.8 1941.64
   135.1 1939.02   213.6 1936.98   223.4 1935.77   246.3 1929.53   262.7 1926.94
   305.2  1924.3  328.011924.279   354.3 1924.71     4031922.658  421.191922.228
   449.2 1923.67     495 1921.29   517.9  1918.8   527.7 1916.84   550.6 1917.33
   557.2 1918.04   560.4 1919.79     567 1925.26   576.8 1930.82   622.6 1945.71
     711 1960.28   766.7 1972.96   773.3 1975.32   786.4 1981.94   802.8 1991.95
#Mann= 7 ,-1 , 0
       0     .12       0    55.5     .06       0  328.01     .12       0
     403    .016       0  421.19     .12       0   517.9    .045       0
   560.4     .12       0
Bank Sta=517.9,560.4
XS Rating Curve= 0 ,0
Exp/Cntr=0.3,0.1

Type RM Length L Ch R = 1 ,96.9    ,107.9,96.9,85.5
XS GIS Cut Line= 3
     2179992.114      235797.015       2180168.2      235323.447
     2180146.498      235047.839
#Sta/Elev= 30
       0 1934.59      23 1933.57    42.6 1929.21    65.6 1925.39   114.8  1922.5
   170.6 1921.39   206.7 1921.55   246.1 1920.18  311.84 1919.12  341.861919.084
   380.6 1919.26   387.1 1917.97     397 1914.66   410.1 1912.97   423.2 1913.29
   429.8 1914.48   436.4 1917.01   446.2 1924.24   452.8 1927.31   485.6 1934.51
     528 1941.04   576.8 1946.94   596.3 1949.95   606.1 1950.43   664.6    1958
   710.2 1966.87   723.2 1970.68   736.2 1976.88   762.2 1991.98   781.7 2005.24
#Mann= 5 ,-1 , 0
       0     .06       0  311.84    .016       0  341.86     .12       0
     397    .045       0   429.8     .12       0
Bank Sta=397,429.8
XS Rating Curve= 0 ,0
Exp/Cntr=0.3,0.1

Chan Stop Cuts=-1
Use User Specified Reach Order=0
Composite Channel Slope=5
